HEC-RAS study RedCreek.prj: RedCreek

--- RedCreek.g01 (geometry) --- (continued)

Type RM Length L Ch R = 1 ,731.5878,46.35,52.4,54.51
XS GIS Cut Line= 3
     627637.7551    4319950.7871     627616.9429    4320031.0395
     627611.4415    4320089.7312
#Sta/Elev= 30
       0  656.34    6.14  654.06   15.35  649.23   27.64  642.43   30.71   640.8
   33.78  639.27   36.85  639.12   39.92  637.51   46.06  633.57   49.13  632.08
    52.2  631.64   55.27  631.47   64.48  630.41   70.62  629.99    73.7  629.61
   82.91  628.43   85.85  627.86    88.8  627.11   91.75  626.62    94.7  626.84
   97.64  627.45  100.59  627.98  103.54  630.41  112.38  637.96  121.22  645.61
  124.17  648.01  127.12  650.14  130.07  650.61  133.01  651.97  141.86   657.3
#Mann= 3 , 0 , 0
       0      .1       0    88.8      .1       0   97.64      .1       0
Bank Sta=88.8,97.64
XS Rating Curve= 0 ,0
Exp/Cntr=0.3,0.1

Type RM Length L Ch R = 1 ,679.1873,37.17,39.11,40.04
XS GIS Cut Line= 3
     627604.1216    4319951.7738     627571.5778    4320016.8614
     627535.0652    4320075.2021
#Sta/Elev= 30
       0  647.79    3.03   646.3     9.1  644.49   12.13  642.96   15.16  641.68
   18.19  640.02   24.26  637.04   27.29   635.4   33.35  631.58   36.39  630.22
   39.42  629.78   45.48  629.61   66.71  627.56   72.77  626.88   75.76  626.14
   81.75  625.17   84.74  624.71   87.73  624.99   90.72  625.46   93.72   626.5
   96.71  627.85    99.7  629.68  105.69  633.66  108.68  635.43  114.66  638.31
  117.66  639.23  120.65  639.86  126.63  642.03   138.6  645.38  141.59  646.05
#Mann= 3 , 0 , 0
       0      .1       0   81.75      .1       0   90.72      .1       0
Bank Sta=81.75,90.72
XS Rating Curve= 0 ,0
Exp/Cntr=0.3,0.1

Type RM Length L Ch R = 1 ,640.08  ,92.71,91.44,89.78
XS GIS Cut Line= 3
     627569.6028    4319938.3482     627541.8756    4319994.4519
     627491.6975    4320046.4991
#Sta/Elev= 28
       0  648.43    2.98  646.87   11.92  642.54   23.84  636.56   26.82  635.14
    29.8  634.75   38.74  629.83   41.72  628.58    44.7  628.03   50.66   627.9
   53.64  627.62   56.62  626.88    59.6  625.77   62.58  624.29   65.59  622.98
   68.61   622.3   71.62  621.51   74.63  622.19   77.64  624.69   80.66   626.7
   83.67  628.23   86.68  629.55    92.7  632.03  107.77  637.99  110.78  639.38
   116.8  640.78  128.85  645.71  134.88  647.78
#Mann= 3 , 0 , 0
       0      .1       0   68.61      .1       0   74.63      .1       0
Bank Sta=68.61,74.63
XS Rating Curve= 0 ,0
Exp/Cntr=0.3,0.1

Type RM Length L Ch R = 1 ,548.64  ,85.4,91.44,96.52
XS GIS Cut Line= 3
     627481.8206    4319911.1232     627450.7459    4319973.2728
     627428.8908    4320031.8865
#Sta/Elev= 25
       0  648.06    3.02   646.7    6.04  645.79   12.08  641.05   15.11  638.87
   18.13  636.79   27.19  630.75   36.25  624.35   39.27  622.95   45.32  622.53
   48.34   622.1    57.4  619.91   60.42  619.08   63.44  618.07   66.46  617.59
   69.49  617.79   72.46  619.02   78.42  620.88    81.4  622.58   93.32  628.64
  105.23  635.28  111.19  637.74  114.17  638.46  117.15   640.1  132.04  648.65
#Mann= 3 , 0 , 0
       0      .1       0   63.44      .1       0   69.49      .1       0
Bank Sta=63.44,69.49
XS Rating Curve= 0 ,0
Exp/Cntr=0.3,0.1

Type RM Length L Ch R = 1 ,457.2   ,89.75,91.44,92.7
XS GIS Cut Line= 2
     627433.3271    4319883.0389     627339.6302    4319937.0958
#Sta/Elev= 30
       0  638.21    9.01  633.38   15.02  630.37   18.03  628.56   24.04  623.98
   27.04  622.02   30.05  620.63   33.05  619.98   36.06  619.56   39.06  616.51
   45.07  612.28   48.08  610.03   51.08  608.12    52.1  607.82   54.09  607.23
   57.09  607.37    60.1  607.77   66.11  609.54   69.11   610.9   72.11  613.06
   75.12  615.47   84.13  622.42   87.14  625.48   90.14  628.89   93.15  631.13
   96.15  633.24   99.16  634.57  102.16  636.63  105.17  638.59  108.17  640.08
#Mann= 3 , 0 , 0
       0      .1       0    52.1      .1       0    60.1      .1       0
Bank Sta=52.1,60.1
XS Rating Curve= 0 ,0
Exp/Cntr=0.3,0.1

Type RM Length L Ch R = 1 ,365.76  ,93.85,91.42,89.98
XS GIS Cut Line= 2
     627398.6403    4319819.0153     627298.3951    4319843.3067
#Sta/Elev= 30
       0   629.7    6.07  626.25     9.1  622.74   21.24  615.25   24.27  614.09
    27.3  613.55   30.34  611.59   33.37  609.44    36.4  607.74   39.44  606.55
   42.47  605.88   48.54  605.06   51.57  603.96   54.61  602.59   57.64   602.3
   60.67  602.53   63.71  603.02   66.74  603.72   69.78  604.66   72.81  605.97
   75.84  608.68   78.88  610.44   81.91  612.47   84.94  614.76   87.98  617.23
   91.01  619.73   94.05  622.64   97.08  625.84  100.11  627.93  103.15  629.32
#Mann= 3 , 0 , 0
       0      .1       0   54.61      .1       0   60.67      .1       0
Bank Sta=54.61,60.67
XS Rating Curve= 0 ,0
Exp/Cntr=0.3,0.1

Type RM Length L Ch R = 1 ,274.3365,94.77,91.46,89.36
XS GIS Cut Line= 2
     627368.3815    4319713.2151     627266.5167    4319776.7152
#Sta/Elev= 30
       0  630.32       3  628.25       6   625.4       9  623.02   18.01  618.09
   24.01  615.57   27.01   613.9   30.01  611.91   33.01  609.12   36.01   607.5
   39.01  606.25   42.01  605.58   45.01  604.55   48.01  602.83   54.02  598.21
   57.02  596.44   60.02  596.29   63.15  597.02   72.02  598.84   75.02  600.17
   81.02  604.08   84.03   606.3   87.03  609.27   93.03   613.3   96.03  614.35
   99.03  615.65  108.03  621.33  111.03  623.88  114.03  626.16  120.04   629.6
#Mann= 3 , 0 , 0
       0      .1       0   57.02      .1       0   63.15      .1       0
Bank Sta=57.02,63.15
XS Rating Curve= 0 ,0
Exp/Cntr=0.3,0.1

Type RM Length L Ch R = 1 ,182.8766,88.26,91.44,94.99
XS GIS Cut Line= 3
       627295.44    4319626.7363     627265.6373    4319667.7448
     627222.7501    4319737.4135
#Sta/Elev= 30
       0  630.64    2.98  627.24    5.96  623.13    8.95  620.42   11.93  617.41
   14.91  614.82   17.89  611.96   23.86  608.71   26.84  605.94   29.82     604
   35.78   602.3   38.77  600.86   41.75  599.28   44.73  597.42   47.71  594.72
   50.69  592.54   52.38   591.7   53.72  591.02   56.75  591.11   59.78  591.65
   62.81  591.83   65.84  592.25   68.87  593.41   74.93  596.56   87.05  602.58
   93.11  605.77   102.2  611.08  105.23   612.3  117.36  619.88  132.51  629.81
#Mann= 3 , 0 , 0
       0      .1       0   52.38      .1       0   59.78      .1       0
Bank Sta=52.38,59.78
XS Rating Curve= 0 ,0
Exp/Cntr=0.3,0.1

Type RM Length L Ch R = 1 ,91.44006,57.38,65.84,67.65
XS GIS Cut Line= 4
     627257.8075    4319579.9861     627217.5869    4319597.3657
     627183.8829    4319621.1973     627143.5327    4319667.3534
#Sta/Elev= 30
       0  630.27    2.92  627.42    5.84  625.15   23.37  613.62   26.29  610.69
   35.05  606.22   46.76  599.51   52.66   594.6   55.61  592.97   61.51  591.32
   64.45  590.03   70.35  586.03    73.3  584.92   76.25   585.1   82.14  586.29
   85.09  587.59   88.16  590.17   91.22  593.13   94.29  595.19   97.35  596.88
  100.42   599.7  103.49  602.02  106.55  604.25  109.62  605.97  112.68  608.38
  124.94  615.74   137.2  624.48  140.27  625.38  143.33  627.81   146.4   631.3
#Mann= 3 , 0 , 0
       0      .1       0   70.35      .1       0   82.14      .1       0
Bank Sta=70.35,82.14
XS Rating Curve= 0 ,0
Exp/Cntr=0.3,0.1

Type RM Length L Ch R = 1 ,25.60198,4.05,9.44,5.97
XS GIS Cut Line= 6
     627257.3831    4319570.9937     627210.5517    4319554.5895
     627166.8954    4319562.7916      627153.137    4319563.0562
     627136.4683    4319573.3749     627113.6093    4319631.5799
#Sta/Elev= 30
       0  631.27    8.76  626.69   14.59   622.5   17.51  620.36   23.35  614.32
   26.27  612.05   35.03  609.32   43.78  601.85   49.62  597.66   58.82  596.11
   64.95  594.17   77.21  591.81   80.28  590.64   83.34  588.27   86.41  586.66
    91.9  584.73  102.19  582.98  105.03  581.17  106.72  580.91  108.41  581.03
  119.67  584.64  126.01  587.17  131.09   590.7  134.07  592.08  137.05  594.39
     143  600.35  148.96  604.68  160.87  611.96  166.82  614.18  190.65  629.68
#Mann= 3 , 0 , 0
       0      .1       0    91.9      .1       0  119.67      .1       0
Bank Sta=91.9,119.67
XS Rating Curve= 0 ,0
Exp/Cntr=0.3,0.1

Type RM Length L Ch R = 1 ,16.16594,2.67,16.17,2.45
XS GIS Cut Line= 6
     627259.4998    4319568.3479     627211.0809    4319551.1499
     627164.2496    4319559.6166     627141.4954    4319557.4999
      627130.912    4319569.6708     627109.6405    4319626.9497
#Sta/Elev= 30
       0  632.19    3.02  629.15    9.07  624.79   18.13  617.31   24.18  613.64
    27.2  612.44   39.29   603.1   45.34  597.87   51.38  593.65   60.36   592.2
   63.36  590.74   81.32  588.47   84.31  587.07    90.3  585.01   93.29  584.24
  105.46  583.27  111.59  580.62  116.88  580.35  119.52  580.58  133.92  584.47
  139.07  587.13  141.64  588.83  144.69  591.95  147.75  594.37   150.8  595.34
  156.91  600.82  163.02  605.18   178.3  614.46  184.41  616.81  202.74  629.48
#Mann= 3 , 0 , 0
       0      .1       0    90.3      .1       0  133.92      .1       0
Bank Sta=90.3,133.92
XS Rating Curve= 0 ,0
Exp/Cntr=0.3,0.1

River Reach=Fisher Spring Rn,1
Reach XY= 30
      643409.528     4318141.789     643331.7403    4318093.1056
     643310.6803    4318078.9654     643299.7412    4318076.4722
     643283.3036    4318074.9596     643253.4235    4318067.7056
     643228.5526    4318073.5264     643198.3901    4318080.4056
     643175.1067    4318073.5264     643151.8024    4318064.4657
     643135.9858    4318062.4614      643126.234    4318059.4645
     643071.3898    4318032.7805     643031.7022    4318016.3763
     642992.5438    4317992.0346     642947.6048     4317962.465
     642927.6759    4317949.9583     642864.4852    4317924.6715
      642843.054     4317913.559     642808.4204    4317871.9646
     642723.9912    4317827.8338     642673.1911     4317798.465
     642654.1411     4317785.765     642596.4618    4317764.5983
     642566.2992    4317751.3691     642509.9429     4317766.715
     642486.1303    4317765.9212      642471.049    4317758.2483
     642451.7344    4317750.3108     642425.7667    4317741.9269

Type RM Length L Ch R = 1 ,1096.86 ,91.1,91.4,92.38
XS GIS Cut Line= 3
     643479.9948    4318022.9409     643401.4376     4318149.328
     643355.1112    4318217.6747
#Sta/Elev= 30
       0 1081.16   21.26 1073.89   27.33 1071.06   30.37 1070.63   39.48 1070.76
   45.55 1070.53   54.67 1069.78   69.85 1067.92   91.11 1065.88   97.18 1065.49
  127.55 1064.61  130.59 1064.35  133.13 1063.86  136.66 1063.17   139.7 1063.61
  142.74 1064.46  145.77 1064.86  148.81  1064.6  151.87 1063.99  157.99 1063.75
  161.04 1064.53  167.16 1066.74  185.51 1070.27  191.62 1071.69  194.68 1071.73
  197.74 1072.46   200.8 1072.88  219.15 1076.39  222.21 1077.19  231.38 1080.36
#Mann= 3 , 0 , 0
       0      .2       0  133.13      .2       0  157.99      .2       0
Bank Sta=133.13,157.99
XS Rating Curve= 0 ,0
Exp/Cntr=0.3,0.1

Type RM Length L Ch R = 1 ,1005.465,33.69,30.95,27.97
XS GIS Cut Line= 4
     643440.8364    4317926.6324     643325.3201    4318098.1245
     643307.7168    4318117.6961      643269.386    4318193.3329
#Sta/Elev= 30
       0 1072.17    15.2 1067.24   18.24 1067.14   45.61 1062.23   54.73 1060.94
    66.9  1060.1   79.06 1059.85   88.18 1060.09   94.26 1059.73  130.75  1060.4
  136.83 1059.64  152.04  1059.1  173.32 1057.12  194.61 1056.06  203.73  1055.2
  206.77 1055.41  212.62 1054.75  218.47  1054.6  224.32 1055.08  233.09 1055.34
  245.21 1056.21  257.32 1057.57  260.35 1057.48  284.58 1060.57   287.6 1061.19
  293.66 1063.21  299.72 1063.97  305.77 1065.85  311.83 1068.02  317.89    1071
#Mann= 3 , 0 , 0
       0      .2       0  212.62      .2       0  224.32      .2       0
Bank Sta=212.62,224.32
XS Rating Curve= 0 ,0
Exp/Cntr=0.3,0.1

Type RM Length L Ch R = 1 ,974.5115,5.96,5.21,4.46
XS GIS Cut Line= 4
     643360.3085    4317921.3563     643307.3917    4318059.4691
     643297.8667    4318095.9817     643261.3541    4318184.8818
#Sta/Elev= 30
       0 1070.24    3.02 1070.11   18.11 1065.79   24.15 1064.46   30.18 1063.54
   36.22 1063.01   63.39 1059.38   69.42 1058.93   72.44 1058.47   84.52 1055.82
   93.57 1053.33   96.59  1052.7  102.63 1052.39   114.7 1052.85  132.81 1053.68
  141.87 1053.57  156.61 1053.93  159.51 1053.88  168.22 1053.13  176.93 1052.85
  206.66 1053.59  218.67 1054.41  233.69 1056.16   239.7 1056.46  257.72 1059.34
  260.72 1060.09  266.73 1062.21  269.73 1062.88  272.73 1063.31  281.74 1066.33
#Mann= 3 , 0 , 0
       0      .2       0   96.59      .2       0   114.7      .2       0
Bank Sta=96.59,114.7
XS Rating Curve= 0 ,0
Exp/Cntr=0.3,0.1

Type RM Length L Ch R = 1 ,969.3049,5.8,5.49,5.19
XS GIS Cut Line= 4
     643345.7652     4317925.838     643299.7276    4318063.5539
     643294.1713    4318097.6852     643259.2462    4318183.8072
#Sta/Elev= 30
       0 1068.49    12.1 1064.85   18.15 1063.54   27.23 1062.31   30.25 1061.99
   33.28  1061.9    60.5 1058.02   66.55 1057.41   75.63 1055.45   87.73 1052.53
   90.75 1052.22   93.78 1052.21  108.91 1052.49  127.06 1053.14  136.13 1052.97
  150.97 1053.02  159.62 1052.69  171.14 1052.69  194.78 1053.35  197.78 1053.27
  212.76 1054.33  227.75 1056.18  230.75  1056.1  248.74 1058.99  251.74  1059.6
  254.73 1060.54  263.73 1063.75  266.73    1064  269.72 1064.86  272.72 1065.94
#Mann= 3 , 0 , 0
       0      .2       0   87.73      .2       0  108.91      .2       0
Bank Sta=87.73,108.91
XS Rating Curve= 0 ,0
Exp/Cntr=0.3,0.1

Type RM Length L Ch R = 1 ,963.8105,12.21,13.04,13.88
XS GIS Cut Line= 4
     643334.2447    4317923.6844     643293.7634    4318062.9878
     643289.7947    4318095.1347     643257.2508    4318182.8443
#Sta/Elev= 30
       0 1067.18    3.02  1067.1   15.11 1063.77   18.13 1063.19   30.22 1061.45
   36.27 1060.96   63.47 1056.87   66.49 1056.72   69.51 1056.24   78.58 1054.29
   84.62 1052.73   87.64  1052.1   90.67 1051.92  102.76 1051.79  114.84 1052.09
  126.93 1052.37  139.02 1052.09  148.01 1052.41   153.9 1052.32  171.57 1052.49
  198.58 1052.98  210.65 1053.75  219.71 1054.79  225.74 1055.67  231.78 1056.04
  249.88 1059.05  255.92 1061.02  261.96 1063.37  267.99 1064.42  271.01 1065.56
#Mann= 3 , 0 , 0
       0      .2       0   87.64      .2       0  114.84      .2       0
Bank Sta=87.64,114.84
XS Rating Curve= 0 ,0
Exp/Cntr=0.3,0.1

Type RM Length L Ch R = 1 ,950.7658,12.93,12.66,12.39
XS GIS Cut Line= 2
      643314.401       4317921.7     643254.4727    4318181.6536
#Sta/Elev= 30
       0 1065.45    3.07 1064.43    6.13 1063.71     9.2 1063.35   15.33 1061.51
    18.4 1060.97    36.8 1058.35   39.86 1058.27   67.46 1054.16   73.59 1053.65
   76.66 1053.04   82.79 1051.48   88.92 1051.69  104.26 1051.19  110.39 1051.06
  128.79 1051.32  141.05 1050.86  151.28 1051.17  162.52 1051.79  177.85  1051.8
  202.38 1052.31  211.58 1052.91  226.91 1055.55  229.98 1055.96  233.04 1056.08
  248.37 1059.04  251.44  1060.1  260.64 1063.83  263.71 1063.85  266.77 1065.03
#Mann= 3 , 0 , 0
       0      .2       0  104.26      .2       0  151.28      .2       0
Bank Sta=104.26,151.28
XS Rating Curve= 0 ,0
Exp/Cntr=0.3,0.1

Type RM Length L Ch R = 1 ,938.1049,5.64,5.72,5.8
XS GIS Cut Line= 2
     643296.8083    4317918.1813     643246.0082    4318178.5318
#Sta/Elev= 30
       0 1063.93    12.2 1060.45   15.24  1060.4   21.34  1058.8   42.69 1055.53
   45.73 1055.38   48.78 1054.98   57.93  1053.5   67.08 1052.49   73.18 1051.38
   76.22 1051.01   79.27 1050.72   82.32 1050.64   88.42 1050.84  118.91  1049.9
  131.11 1049.83   143.3 1049.49   149.4 1049.74  164.64 1050.94  176.84 1050.94
  192.09 1051.34  204.28  1051.8  213.43 1052.57  222.57 1053.94  231.72 1055.56
  234.77 1055.65  250.02 1058.64  253.06 1059.77  262.21 1063.62  265.26  1063.7
#Mann= 3 , 0 , 0
       0      .2       0  131.11      .2       0   149.4      .2       0
Bank Sta=131.11,149.4
XS Rating Curve= 0 ,0
Exp/Cntr=0.3,0.1

Type RM Length L Ch R = 1 ,932.3828,10.05,8.03,6
XS GIS Cut Line= 5
     643284.6463    4317917.9004     643264.8025    4318053.2351
     643258.8494     4318082.207     643257.2619    4318107.2102
     643243.3712    4318177.0603
#Sta/Elev= 30
       0 1063.04   12.16 1059.94    15.2 1059.53   21.28 1059.21   39.51 1054.84
   45.59 1053.59   48.63 1053.35   54.71 1052.25   60.79 1051.44   69.91 1050.86
   75.99 1050.24   79.03 1050.27   85.11 1050.69  106.39 1049.78  121.58  1049.4
  133.74 1049.23  148.61 1049.46   163.4 1050.46  174.71 1050.55  191.41 1051.21
  206.25 1051.93  212.18  1052.5  221.09 1053.81  229.99 1055.45  232.96 1055.56
  235.92 1056.03  247.79 1058.29  250.76 1059.22  259.66 1062.95  262.63  1063.7
#Mann= 3 , 0 , 0
       0      .2       0  121.58      .2       0  148.61      .2       0
Bank Sta=121.58,148.61
XS Rating Curve= 0 ,0
Exp/Cntr=0.3,0.1

Type RM Length L Ch R = 1 ,924.3561,6.01,5.17,4.34
XS GIS Cut Line= 4
      643272.729    4317913.7625     643250.9008    4318004.2501
     643255.2665    4318105.8503     643241.3758    4318176.4942
#Sta/Elev= 30
       0 1062.63    6.01 1060.82   18.02 1057.46   30.03 1055.55   39.03 1053.87
   51.05 1052.16   57.05 1051.69   69.06 1050.39   72.06    1050   78.07 1048.81
   81.07 1048.67   84.08  1048.9   87.08 1048.92  111.03 1048.25  128.98 1048.01
  137.95 1048.21  143.93 1048.61  161.88 1049.28  170.85 1049.99  182.81 1050.33
  206.78 1051.79  209.78 1051.77  212.78 1051.94  215.78 1052.22  227.78 1054.06
  236.78 1055.64  242.77 1056.32  251.77 1057.99  254.77 1058.84  266.77 1063.78
#Mann= 3 , 0 , 0
       0      .2       0  111.03      .2       0  137.95      .2       0
Bank Sta=111.03,137.95
XS Rating Curve= 0 ,0
Exp/Cntr=0.3,0.1

Type RM Length L Ch R = 1 ,919.1814,5.84,5.17,4.49
XS GIS Cut Line= 4
     643265.8608    4317913.4687      643238.741    4318001.7735
      643253.981    4318105.5301     643238.1801    4318177.0418
#Sta/Elev= 30
       0 1061.96   11.92 1058.36   23.84 1055.16   26.82 1055.08    29.8 1054.35
   41.72 1052.38   53.64 1050.98    59.6 1050.66   71.52 1049.52    74.5 1049.12
   80.46 1047.76   83.44 1047.42   98.37 1047.31  113.35 1047.11  128.33 1047.32
  137.32 1047.52  164.29 1048.98  173.28 1049.68  185.26 1050.03   200.3 1051.13
  209.45 1051.68   212.5 1051.64  218.61 1052.14  233.86 1054.47  239.97 1055.63
  243.02 1055.79  246.07 1056.19  255.22 1057.96  258.28  1058.9  270.48    1064
#Mann= 3 , 0 , 0
       0      .2       0   98.37      .2       0  128.33      .2       0
Bank Sta=98.37,128.33
XS Rating Curve= 0 ,0
Exp/Cntr=0.3,0.1

Type RM Length L Ch R = 1 ,914.013 ,52.15,56.37,60.59
XS GIS Cut Line= 4
     643257.7443     4317909.699      643226.098    4317995.4074
     643251.7828    4318105.1525     643236.5776    4318174.2829
#Sta/Elev= 30
       0 1061.98   12.18 1058.26   27.41 1053.96   30.45 1053.71   36.55 1052.57
   45.68 1051.47   63.95    1050      67 1049.89   88.32 1046.52   91.36 1046.04
  103.55 1046.41  124.87 1046.29  134.01 1046.39  143.15 1046.68  155.34 1047.81
  161.43 1048.03  170.57 1048.58   179.7 1049.38  191.89 1049.81  207.02 1050.94
  215.87  1051.5  221.77 1051.67  224.72 1051.95  242.42 1054.64  248.31 1055.71
  251.26 1055.71  260.11 1057.39  263.06 1058.03  266.01 1059.05  274.86 1062.76
#Mann= 3 , 0 , 0
       0      .2       0   88.32      .2       0  134.01      .2       0
Bank Sta=88.32,134.01
XS Rating Curve= 0 ,0
Exp/Cntr=0.3,0.1

Type RM Length L Ch R = 1 ,857.6442,22.65,23.23,23.8
XS GIS Cut Line= 2
     643239.6582    4317904.7757     643155.5205    4318190.5263
#Sta/Elev= 30
       0 1060.47    3.07 1059.51    6.14 1059.18    9.21 1058.45   30.71 1052.36
   33.78 1051.54   36.85 1051.05   67.56 1047.84    73.7 1047.43   85.99  1046.2
    95.2 1044.74   98.27 1044.54  104.41 1044.62  110.55 1044.41  135.12 1043.16
  171.97 1042.99  178.11  1043.1  184.26 1043.42  199.61 1045.34  202.68 1045.35
  218.04 1047.54  233.39 1050.25  239.53 1050.86  257.96  1053.9   264.1 1054.79
  270.24 1055.23  273.31 1056.12  279.45 1058.94  294.81 1066.49  297.88 1068.46
#Mann= 3 , 0 , 0
       0      .2       0  135.12      .2       0  178.11      .2       0
Bank Sta=135.12,178.11
XS Rating Curve= 0 ,0
Exp/Cntr=0.3,0.1

Type RM Length L Ch R = 1 ,834.4178,11.41,11.53,11.65
XS GIS Cut Line= 2
     643230.2633    4317900.6656     643124.2974     4318183.638
#Sta/Elev= 30
       0 1060.33    9.16 1057.76   12.21 1057.07   15.26 1056.81   36.63 1050.84
   42.73 1049.46   61.04 1047.48   94.62 1044.35   97.67 1043.93  103.77 1042.44
  106.83 1041.95  109.88 1042.32  112.93  1042.3  122.09 1041.57  125.14 1041.43
  137.35 1041.83  161.76 1041.57  183.13  1041.7  186.18 1041.78  213.65 1044.42
  222.81    1045  228.91 1045.97  247.22 1049.79  253.33 1050.24  274.69 1053.87
  277.75 1054.62  283.85 1057.26   286.9 1057.69  296.06 1062.41  302.16 1066.32
#Mann= 3 , 0 , 0
       0      .2       0  122.09      .2       0  183.13      .2       0
Bank Sta=122.09,183.13
XS Rating Curve= 0 ,0
Exp/Cntr=0.3,0.1

Type RM Length L Ch R = 1 ,822.8911,18.45,17.05,15.65
XS GIS Cut Line= 2
     643225.9943     4317887.474     643111.7362    4318179.0821
#Sta/Elev= 30
       0 1063.24    9.21 1060.65   18.42 1057.72   24.56  1056.1   30.71 1055.04
   42.99 1051.62   55.27  1048.6   61.41 1047.77  101.33 1043.87  119.75 1040.36
  128.96 1040.07  138.17 1040.31  147.39 1040.82  159.67    1041  184.23 1041.01
  190.37 1040.57  196.51 1041.25  218.01 1042.43  233.36 1043.81  236.43 1043.78
  242.57  1044.8  264.07 1049.38  267.14 1049.82  270.21  1049.8   291.7 1053.87
  294.77 1055.04  297.84 1056.61  300.91 1057.67  303.98 1058.27  313.19 1063.52
#Mann= 3 , 0 , 0
       0      .2       0  119.75      .2       0  138.17      .2       0
Bank Sta=119.75,138.17
XS Rating Curve= 0 ,0
Exp/Cntr=0.3,0.1

Type RM Length L Ch R = 1 ,805.843 ,17.81,19.53,21.24
XS GIS Cut Line= 4
     643209.6257    4317891.1405     643142.5537    4318047.1127
       643135.41    4318082.4347     643098.5005     4318174.113
#Sta/Elev= 30
       0 1059.45   24.25 1053.21   30.32 1052.34   39.41 1049.63   51.54  1046.8
    66.7 1045.16   93.99 1041.78  100.05 1041.38  109.15 1040.24  115.21 1039.17
  118.24 1038.72  130.37 1039.25  148.56 1039.57  175.79  1039.6  181.79    1039
   184.8 1039.25   190.8 1040.43  196.81  1040.9   217.8 1041.65  223.79 1042.21
  229.78 1043.23  232.77 1043.29  235.77 1043.74  265.72 1049.91  271.71 1050.47
  283.68 1052.99  286.68 1053.75  289.67  1054.9  298.66 1059.56  304.65 1061.08
#Mann= 3 , 0 , 0
       0      .2       0  115.21      .2       0   184.8      .2       0
Bank Sta=115.21,184.8
XS Rating Curve= 0 ,0
Exp/Cntr=0.3,0.1

Type RM Length L Ch R = 1 ,786.3173,33.09,32.99,32.9
XS GIS Cut Line= 2
     643196.0019    4317885.7257     643073.7641    4318164.3325
#Sta/Elev= 30
       0 1057.15    6.15 1056.19   18.44 1053.18    33.8 1049.77   39.95 1048.94
   58.39 1044.79   67.61 1043.69   76.83 1042.92  104.49 1039.99  110.63 1039.57
  113.71 1039.18  119.85 1037.87  122.93  1037.5  129.07 1037.93  153.66 1037.89
  175.17 1037.27  184.39  1036.9  187.46 1037.13  193.61 1037.72  212.05 1038.73
  221.27 1039.72  227.41  1040.7  245.85 1044.95  248.93 1045.08     252 1045.63
  279.66  1051.3  282.73 1051.39   285.8 1052.12  291.95 1054.08  304.24 1058.84
#Mann= 3 , 0 , 0
       0      .2       0  175.17      .2       0  187.46      .2       0
Bank Sta=175.17,187.46
XS Rating Curve= 0 ,0
Exp/Cntr=0.3,0.1

Type RM Length L Ch R = 1 ,753.324 ,22.54,22.45,22.35
XS GIS Cut Line= 2
     643161.8706    4317876.2007     643045.1891    4318150.8387
#Sta/Elev= 30
       0 1054.47   18.27 1049.16   21.31 1048.98   36.54 1045.62   51.76 1042.71
   54.81 1042.59   63.94 1041.14   73.08 1040.24   85.26 1038.35  100.48 1036.51
  124.84 1034.57  130.93 1034.35  152.24 1034.76  164.42 1034.51  173.56 1034.77
  179.65 1034.48  182.69 1034.92  185.74 1035.46  191.83 1035.83  197.92 1035.85
   210.1 1037.04  225.32 1039.81  228.36 1039.82  231.41 1040.37  261.86 1046.46
   264.9 1046.51  267.95 1047.11  274.04 1048.88  295.35 1056.11   298.4 1056.16
#Mann= 3 , 0 , 0
       0      .2       0  124.84      .2       0  182.69      .2       0
Bank Sta=124.84,182.69
XS Rating Curve= 0 ,0
Exp/Cntr=0.3,0.1

Type RM Length L Ch R = 1 ,730.8785,34.15,34.8,35.45
XS GIS Cut Line= 2
      643141.151    4317861.9857     643026.8201    4318140.3153
#Sta/Elev= 30
       0 1052.63    3.07 1051.72    6.14  1051.4   15.35 1048.98   36.84 1044.29
   39.91 1044.16   55.27 1040.89   73.69 1037.53   76.76 1037.34   85.97  1036.1
  104.39 1034.34  141.24 1033.16  147.38 1032.45  150.45 1032.07  159.66 1032.52
  171.94 1032.52  184.22 1032.16  189.49 1032.44  202.64 1033.71  208.79 1034.64
  211.86 1034.78  214.93 1035.14  245.63 1040.96   248.7 1041.03  251.77 1041.48
  267.12 1044.65   279.4 1047.51  282.47 1047.51  291.69 1050.38   300.9 1053.55
#Mann= 3 , 0 , 0
       0      .2       0  147.38      .2       0  189.49      .2       0
Bank Sta=147.38,189.49
XS Rating Curve= 0 ,0
Exp/Cntr=0.3,0.1

Type RM Length L Ch R = 1 ,696.0811,31.98,32.59,33.19
XS GIS Cut Line= 2
      643115.833    4317868.2632      642984.864    4318125.4387
#Sta/Elev= 30
       0 1047.29    3.07 1047.12    6.14 1046.58   36.84 1040.67   42.98    1040
   52.19 1037.94   70.62 1034.48   73.69 1034.08    82.9 1033.41  104.39 1032.32
  110.53 1031.29  116.67 1030.96  135.09 1030.18  156.58 1029.64  165.79  1029.2
  171.93 1029.46  181.14 1030.55  187.29  1030.7   196.5 1031.45  199.57 1031.84
  221.06 1035.45  224.13 1035.41  230.27 1036.38  236.41 1037.49  245.62 1039.48
  254.83 1040.89   257.9    1041  260.97 1041.51  282.46 1046.96   288.6 1048.99
#Mann= 3 , 0 , 0
       0      .2       0  156.58      .2       0  171.93      .2       0
Bank Sta=156.58,171.93
XS Rating Curve= 0 ,0
Exp/Cntr=0.3,0.1

Type RM Length L Ch R = 1 ,663.4952,23.62,23.9,24.17
XS GIS Cut Line= 2
     643095.1954    4317864.2944     642945.9701    4318109.5636
#Sta/Elev= 30
       0 1045.29    6.11 1044.07   18.33 1042.17   30.54 1039.61    33.6 1039.15
    39.7 1037.59   45.81 1036.39   51.92 1035.66    73.3 1031.39   85.52 1030.45
   94.68 1029.97  134.39 1028.47  140.49 1028.03  157.69 1027.39  164.93  1026.9
  171.04 1027.32  174.09  1027.7  195.47 1028.94  201.58  1029.6  207.69 1029.98
  222.96 1032.52  241.28 1035.91  247.39 1036.39   253.5 1037.25  259.61 1038.45
  262.66 1039.26  268.77 1041.17  280.99 1045.45  284.04 1045.86   287.1 1046.55
#Mann= 3 , 0 , 0
       0      .2       0  157.69      .2       0  171.04      .2       0
Bank Sta=157.69,171.04
XS Rating Curve= 0 ,0
Exp/Cntr=0.3,0.1

Type RM Length L Ch R = 1 ,639.5986,93.16,91.54,89.92
XS GIS Cut Line= 2
     643077.6509    4317857.7524     642921.2966    4318095.7637
#Sta/Elev= 30
       0 1044.11   21.43 1039.68    24.5 1039.14   27.56 1038.91   33.68 1037.65
   39.81 1035.99   58.18 1032.05   76.55 1028.66   79.61 1028.31   82.68  1028.2
    88.8 1027.45  104.11 1026.48  128.61 1025.72  150.04 1024.37  156.17 1023.91
  159.23 1023.97  162.29 1024.37  168.41 1025.06  180.66 1025.94  186.79  1025.9
   202.1 1027.13  211.28  1028.6  220.47 1030.39  226.59 1030.82  244.97 1033.93
  254.15 1035.72  263.34  1037.8   266.4 1037.91  272.53 1040.55  284.77 1045.11
#Mann= 3 , 0 , 0
       0      .2       0  150.04      .2       0  162.29      .2       0
Bank Sta=150.04,162.29
XS Rating Curve= 0 ,0
Exp/Cntr=0.3,0.1

Type RM Length L Ch R = 1 ,548.0592,87.22,91.25,95.27
XS GIS Cut Line= 2
      642964.409     4317812.244     642871.2146    4318046.3231
#Sta/Elev= 30
       0 1035.02    9.22 1033.55   24.58 1029.69   27.65 1029.43   36.87  1026.7
   49.16 1022.71   52.23 1021.82   55.31 1021.14   76.81 1019.07   86.03 1018.01
   122.9 1016.06  135.19 1015.14  138.26  1014.7  141.34 1014.54   146.5 1015.19
  150.55 1015.65  159.77 1016.35  162.84  1016.2  165.92 1016.52  178.21 1018.46
  193.57 1021.12  196.64 1021.53  199.72 1021.55  205.86 1022.59  212.01 1023.85
  227.37  1027.4  233.51 1027.97  242.73 1030.01  248.88 1032.12  251.95 1033.42
#Mann= 3 , 0 , 0
       0      .2       0  135.19      .2       0   146.5      .2       0
Bank Sta=135.19,146.5
XS Rating Curve= 0 ,0
Exp/Cntr=0.3,0.1

Type RM Length L Ch R = 1 ,456.813 ,94.43,91.27,88.11
XS GIS Cut Line= 2
     642903.7829    4317842.3615     642742.4266     4317976.715
#Sta/Elev= 30
       0 1018.23    3.04 1017.15    6.09 1016.68    9.13 1015.52   12.17 1014.57
   24.34 1011.23   27.39 1010.73   33.47 1010.16   39.56 1009.21   60.86 1007.02
   66.95 1006.14   69.99 1005.44    85.2 1003.81   91.29 1002.88   94.33 1002.36
   97.23  1002.3  100.42 1002.73  112.59 1004.38  115.63 1004.63  118.68 1005.14
  121.72 1005.15  130.85 1006.25  139.98 1007.16  152.15 1008.14  158.24 1008.45
  173.45 1009.55   176.5 1009.68  179.54 1009.63   197.8 1013.94  209.97 1017.39
#Mann= 3 , 0 , 0
       0      .2       0   91.29      .2       0  100.42      .2       0
Bank Sta=91.29,100.42
XS Rating Curve= 0 ,0
Exp/Cntr=0.3,0.1

Type RM Length L Ch R = 1 ,365.5449,29.51,29.71,29.92
XS GIS Cut Line= 2
     642812.0087    4317751.9189     642707.2335    4317949.8276
#Sta/Elev= 30
       0 1009.01     9.2 1005.94   12.27 1005.06   15.34 1004.31   21.47 1003.17
   27.61 1002.26   36.81 1001.25   55.22  997.96   58.28  997.92   76.69  994.83
   79.76  994.44   104.3  993.02  107.36  992.42  110.43  991.83   113.5  992.56
  116.57  993.37  119.64  993.83  128.84  994.24  131.91  994.11  144.18     995
  153.38  995.99  165.65  997.67  171.78  997.91  180.99   999.2  187.12  999.69
  190.19 1000.14  205.53 1004.06  208.59 1004.18   217.8 1006.53  223.93 1008.36
#Mann= 3 , 0 , 0
       0      .2       0  107.36      .2       0   113.5      .2       0
Bank Sta=107.36,113.5
XS Rating Curve= 0 ,0
Exp/Cntr=0.3,0.1

Type RM Length L Ch R = 1 ,335.8305,31.7,31.86,32.01
XS GIS Cut Line= 2
     642780.7904    4317752.4548     642680.7777    4317930.2552
#Sta/Elev= 27
       0 1003.45   12.18 1000.34   21.31   997.8   24.36  997.17    27.4  996.92
   33.49  995.59   36.54  995.22   42.63  994.15    60.9  991.69   66.98  991.25
   82.21  989.73   85.25  989.35   88.16   988.8   91.34   988.3   94.39  988.38
  100.48  988.95  106.57  988.97  121.79  989.73  137.01  990.98  140.06  990.86
  146.15  991.36  167.46  994.51  170.51  995.04  173.55  995.82   176.6  996.32
  179.64  996.58     204 1004.11
#Mann= 3 , 0 , 0
       0      .2       0   88.16      .2       0  106.57      .2       0
Bank Sta=88.16,106.57
XS Rating Curve= 0 ,0
Exp/Cntr=0.3,0.1

Type RM Length L Ch R = 1 ,303.9727,30.24,30.2,30.15
XS GIS Cut Line= 2
     642750.6279    4317744.5173     642652.9964    4317910.4114
#Sta/Elev= 30
       0  998.12    6.11  996.92    9.17  995.97   18.33  994.02    27.5  992.61
   39.72  990.25   42.78  989.79   51.94  988.13   58.05  986.43   64.16  985.71
   67.22  985.46   70.27  985.32   76.39  985.34   79.44  984.93    82.5  984.61
   85.55  984.06   88.61  984.32   91.66  984.94   94.72  985.21  106.94  985.29
  113.05  985.02  119.16  985.14  122.22  984.94  125.27  985.03  131.38  985.64
  152.77  988.51  161.94  989.08  164.99  989.67  177.21  993.45  192.49  997.75
#Mann= 3 , 0 , 0
       0      .2       0   79.44      .2       0  125.27      .2       0
Bank Sta=79.44,125.27
XS Rating Curve= 0 ,0
Exp/Cntr=0.3,0.1

Type RM Length L Ch R = 1 ,273.7743,29.55,29.12,28.69
XS GIS Cut Line= 2
     642721.2126    4317734.0548     642627.8584    4317894.7941
#Sta/Elev= 30
       0  991.04    6.09  989.12    9.14  988.43   18.28  986.52   27.43  984.74
   30.47  983.88   33.52  983.56   36.57  982.86   39.61  982.33   45.71  981.42
    51.8  980.75   60.94  980.09   70.09  979.64   73.13  979.17   76.18   978.6
   79.23  978.76   82.28  979.16   97.51  979.42  103.61  979.19   109.7  979.32
  121.89  979.76  137.13  981.18  140.17  980.87  143.22  981.02  158.46     983
   161.5  983.76  170.65  986.76  173.69  987.47  176.74  987.34  185.88  990.12
#Mann= 3 , 0 , 0
       0      .2       0   73.13      .2       0   109.7      .2       0
Bank Sta=73.13,109.7
XS Rating Curve= 0 ,0
Exp/Cntr=0.3,0.1

Type RM Length L Ch R = 1 ,244.652 ,32.3,31.64,30.97
XS GIS Cut Line= 2
      642689.509     4317723.086     642602.9901    4317892.1551
#Sta/Elev= 29
       0  984.89    3.06   984.2    9.19  983.18   30.63  977.94   36.76  976.59
   39.82  976.14   52.08  974.98   55.14  974.45   61.26  973.93   67.21  972.57
   70.45  972.05   73.52  972.39   76.58  972.98   79.64  972.86   94.96  973.94
  110.28   974.9  113.34  975.07  122.53  975.31  134.78  975.89  140.91  976.28
   150.1  977.14  153.16  977.02  159.29  977.96  162.35  978.52  165.41  979.18
  168.48  980.01   174.6  982.11  186.86  987.17  189.92  987.32
#Mann= 3 , 0 , 0
       0      .2       0   67.21      .2       0   76.58      .2       0
Bank Sta=67.21,76.58
XS Rating Curve= 0 ,0
Exp/Cntr=0.3,0.1

Type RM Length L Ch R = 1 ,213.0166,30.51,30.22,29.93
XS GIS Cut Line= 2
     642657.7589    4317701.6547     642578.3838    4317894.5363
#Sta/Elev= 30
       0   983.4    6.13  982.22   15.34  979.16    18.4  978.37   27.61  974.79
   33.74  972.71   36.81  972.34   46.01  969.61   58.28  967.71   70.55  967.06
   73.61  966.39   76.68  965.18   79.75  963.41   82.82  963.77   85.27  964.82
   88.95  966.05  101.22  968.17  104.29  968.31  107.36  967.93  119.62  970.07
  125.76  970.91  134.96  971.88   141.1  972.12   168.7  975.28   177.9  975.63
  180.97  976.16   187.1   978.1  199.37  983.77  205.51  986.27  208.58  986.74
#Mann= 3 , 0 , 0
       0      .2       0   76.68      .2       0   85.27      .2       0
Bank Sta=76.68,85.27
XS Rating Curve= 0 ,0
Exp/Cntr=0.3,0.1

Type RM Length L Ch R = 1 ,182.7951,101.25,91.74,91.18
XS GIS Cut Line= 2
     642628.9167    4317684.1854     642550.5999    4317895.8525
#Sta/Elev= 30
       0  982.23    9.15  977.83   15.25  975.43    24.4   972.5    30.5  971.44
   39.65  968.56   45.75  966.89    54.9  963.59   57.95  962.71      61  962.38
   64.05  961.84   70.15  959.54   76.25  957.96   82.35  955.33    85.4   954.5
   88.45  954.63   91.67  955.43   94.55  955.28  125.05  964.54  128.09  965.24
  131.14  965.26  134.19   966.1  137.24  966.71  158.59  969.32  164.69  969.27
  189.09  971.69  195.19  971.45  198.24  971.85  201.29  972.74  225.69  982.75
#Mann= 3 , 0 , 0
       0      .2       0   82.35      .2       0   91.67      .2       0
Bank Sta=82.35,91.67
XS Rating Curve= 0 ,0
Exp/Cntr=0.3,0.1

Type RM Length L Ch R = 1 ,91.05302,41.6,41.6,41.6
XS GIS Cut Line= 6
     642569.6499     4317657.727     642507.1709    4317743.8898
      642508.973    4317757.1786     642514.3894     4317774.912
     642525.1361    4317796.5155     642538.9582    4317876.8024
#Sta/Elev= 30
       0  972.19    3.04  971.47   12.16   968.6   24.33  965.29   30.41  963.37
    66.9  956.71   69.94  955.83   79.06  953.94   85.15  953.03  100.35  948.83
  109.11  945.78  117.16  943.29  119.84  943.31  121.93  942.82   126.9  940.75
  129.78  939.79  132.66  940.02  134.16  940.63  147.46  946.71  150.48  947.09
  165.56  953.32  174.61  956.12  177.63  957.33  183.66  958.65   189.7  960.79
   207.8  964.45  210.82  964.58  234.96  970.07  240.99  970.92  244.01  971.62
#Mann= 3 , 0 , 0
       0      .2       0   126.9      .2       0  134.16      .2       0
Bank Sta=126.9,134.16
XS Rating Curve= 0 ,0
Exp/Cntr=0.3,0.1

Type RM Length L Ch R = 1 ,50      ,41,50,38
XS GIS Cut Line= 4
642510.312868476 4317703.4604645642473.8450398814317748.25247136
642468.8901718654317779.96362666642491.9256720484317863.12856687
#Sta/Elev= 30
       0 952.625   2.093 952.116   6.962 949.999  10.418 949.209  24.164 946.404
  41.047   943.8  45.916 942.513  50.061 941.741  64.164 936.912  70.387 934.024
  73.498 933.897   76.61 933.357  80.972 933.907  82.833 934.184  89.856 936.032
  92.226 937.038  95.416 938.644 101.796 942.272 104.986 942.354 108.176 944.214
 111.366 945.634 120.936  948.92 130.507  952.58 133.697 952.697 140.077 954.776
 143.267 955.563 159.217 958.466 162.407  958.73 168.787 960.291 176.152 961.804
#Mann= 3 , 0 , 0
       0      .2       0  73.498      .2       0  80.972      .2       0
Bank Sta=73.498,80.972
XS Rating Curve= 0 ,0
Exp/Cntr(USF)=0,0
Exp/Cntr=0.3,0.1

River Reach=Gandy Run       ,1
Reach XY= 30
     637221.3776    4315926.2187     637200.8723    4315907.3671
     637194.5884     4315892.815     637185.9895    4315826.3383
     637170.1144    4315772.4293     637171.7681    4315731.0881
     637182.0207    4315720.5047     637186.9817    4315700.9917
     637155.5623    4315640.7988     637154.9009    4315602.4342
     637177.0598    4315572.3378     637183.0129     4315503.546
     637170.7759    4315485.0251     637191.6119    4315437.0693
      637209.802    4315362.9858     637256.1042     4315322.306
     637275.7565    4315281.4163     637278.2631    4315205.2276
     637260.7562    4315160.4174     637258.8144    4315130.9059
     637276.6094     4315064.006     637289.9214    4315055.9444
      637288.185    4315036.5554     637254.7813    4315006.7898
     637202.3913    4315018.9627     637182.2498    4315016.5319
     637115.9715    4314954.2224     637031.3941      4314919.77
     636979.4463    4314877.6254     636956.1954    4314870.4384

Type RM Length L Ch R = 1 ,1371.6  ,86.38,91.44,95.29
XS GIS Cut Line= 4
     637306.8057    4315867.8062     637241.9582     4315901.754
     637191.5243     4315956.612     637138.9689     4315978.719
#Sta/Elev= 30
       0   864.3    12.2  860.42    18.3  857.59   33.55   852.9    42.7  850.85
      61  847.72    67.1  845.53    73.2  844.36   94.06  842.97   97.04  841.22
  100.02  838.51  102.14  837.52     103  837.12  105.98  837.03  111.95  837.61
  129.83  839.27  135.79  839.68  138.77  840.11  141.75  841.08  144.73  842.52
  150.72   845.9  156.72   849.7  159.72  852.09  162.72  855.21  165.72  856.51
  168.72  857.16  180.72  858.44  192.73  860.53  198.73  861.83  204.73  863.56
#Mann= 3 , 0 , 0
       0      .1       0  102.14      .1       0  111.95      .1       0
Bank Sta=102.14,111.95
XS Rating Curve= 0 ,0
Exp/Cntr=0.3,0.1

Type RM Length L Ch R = 1 ,1280.16 ,91.85,91.38,92.13
XS GIS Cut Line= 3
     637281.6462    4315840.8834     637184.2562    4315844.4905
     637052.1437    4315869.1291
#Sta/Elev= 30
       0  854.65    6.09  851.45   21.32  847.08   27.41  844.67   42.64  840.97
   48.73  839.08   82.23   832.9   85.27  832.25   88.32  830.89   94.41   830.2
   97.46  831.01  106.62  836.44  109.67  839.45  112.73  841.02     128  847.19
  131.05  849.06  134.11  849.68  137.16  849.14  140.22  847.95  146.33  844.76
  149.38  842.64  152.43  839.72  155.49  837.33  158.54  836.46   161.6  836.47
  167.71  838.31  173.81  841.77  179.92   843.8  207.41  847.73  231.85  854.47
#Mann= 3 , 0 , 0
       0      .1       0   88.32      .1       0   97.46      .1       0
Bank Sta=88.32,97.46
XS Rating Curve= 0 ,0
Exp/Cntr=0.3,0.1

Type RM Length L Ch R = 1 ,1188.777,93.59,91.5,90.83
XS GIS Cut Line= 2
     637272.4098    4315742.7903     637103.3864    4315763.7478
#Sta/Elev= 30
       0   855.2    6.08  852.21   18.25   848.2   21.29  846.99   24.33  845.26
   42.58  839.47   45.62  837.66   54.75  834.93   63.87  832.44   66.91  830.77
   69.95  830.04   79.08  828.74   82.12  827.78   85.16  826.46    88.2  825.49
   94.28  825.29   97.32  824.85  100.37  823.97  103.41  823.11  106.45  823.19
  112.53  827.98   124.7  833.92  127.74  836.23  130.78  838.31  133.82  839.75
  145.99  844.96  152.07  849.23  158.15  851.93  161.19  852.96  170.32   855.3
#Mann= 3 , 0 , 0
       0      .1       0  100.37      .1       0  106.45      .1       0
Bank Sta=100.37,106.45
XS Rating Curve= 0 ,0
Exp/Cntr=0.3,0.1

Type RM Length L Ch R = 1 ,1097.275,84.7,91.43,97.49
XS GIS Cut Line= 3
     637248.4914     4315633.279     637169.4435    4315674.0651
     637092.1223    4315706.3042
#Sta/Elev= 30
       0  847.07    3.07  845.81    6.13  843.47     9.2  842.18   27.61  835.22
   33.74  832.11   36.81   830.9   55.21  824.85   58.28   822.9   67.48  820.14
   70.55  818.82   76.68  815.27   79.75  814.44   85.88  815.09   91.94  815.92
  100.92  817.78  103.91   818.8   106.9  820.12  109.89  820.97  115.88  822.13
  118.87  823.28  124.85  824.42  127.84  825.53  130.84  826.99  136.82  829.48
  148.79  834.96  151.78  837.11  154.77  838.75  169.73  845.29  172.72  846.44
#Mann= 3 , 0 , 0
       0      .1       0   76.68      .1       0   85.88      .1       0
Bank Sta=76.68,85.88
XS Rating Curve= 0 ,0
Exp/Cntr=0.3,0.1

Type RM Length L Ch R = 1 ,1005.84 ,101.14,91.44,83.95
XS GIS Cut Line= 4
     637231.1157    4315612.6931     637191.4276    4315608.0508
      637144.284    4315573.3406     636943.6908    4315619.7852
#Sta/Elev= 30
       0  837.96    3.07  836.44    6.15  833.76    9.22  831.91   21.52  826.01
   27.66  821.71   48.74  811.56    66.3  808.44   72.16  808.06   75.08  808.48
   83.87  811.83   89.72  813.57   92.65  814.09  113.87  815.47  123.09  816.76
  135.38   820.6  141.53   823.6  153.82  827.79  159.96  829.71  163.04  830.27
  199.92  831.76  239.87  832.32  246.01  833.27  255.23  833.62  264.45  832.98
   270.6  832.16  285.96  831.47  289.04  831.82  295.18  833.98   304.4   836.5
#Mann= 3 , 0 , 0
       0      .1       0    66.3      .1       0   75.08      .1       0
Bank Sta=66.3,75.08
XS Rating Curve= 0 ,0
Exp/Cntr=0.3,0.1

Type RM Length L Ch R = 1 ,914.4   ,86.34,91.44,102.73
XS GIS Cut Line= 6
     637248.6773    4315478.7277     637194.7414    4315488.5168
     637185.0259    4315499.1869     637177.6225    4315505.5057
     637174.0311    4315505.0202     637040.5285    4315541.9976
#Sta/Elev= 30
       0  828.39    3.05  827.42    6.09  825.46   24.36  819.68   27.41  817.61
   30.45  816.35   36.54  814.26   45.68  811.61   51.77  808.25   54.82  807.09
   63.48   804.8   71.68  802.08   74.11  801.26   76.55  801.35   78.98  801.87
   97.66  805.11  100.67  806.39  103.69  807.08  118.74  809.19  127.78  811.64
  139.82  815.45  142.83  816.53  145.85  818.07  154.88   820.5  157.89   820.9
  163.92  821.21  172.95  822.84  191.02  824.99   212.1  827.31  221.13  828.07
#Mann= 3 , 0 , 0
       0      .1       0   71.68      .1       0   78.98      .1       0
Bank Sta=71.68,78.98
XS Rating Curve= 0 ,0
Exp/Cntr=0.3,0.1

Type RM Length L Ch R = 1 ,822.96  ,86.45,91.44,99.46
XS GIS Cut Line= 5
     637256.9916    4315431.0865     637198.0266    4315419.4414
     637193.9291    4315418.3513     637165.8467    4315407.5851
     637036.5068    4315435.7407
#Sta/Elev= 30
       0  818.78    6.01  816.56    9.02  815.15   12.02  814.52   24.04  810.35
   30.05  807.51   45.08  802.79   48.08  801.16    60.1  796.62   62.22   796.2
   64.34  796.14   67.35  796.91   70.36  798.55   73.37  799.42   76.37  799.72
   94.42  799.42   97.43  799.84  100.44   800.7  109.46  804.17  112.47  806.59
  115.48  808.21  118.49  809.28  121.49  810.03   124.5  810.46  148.57  812.23
  154.59  812.87  169.63  813.72  175.65  814.66  205.73  818.09  226.79  818.76
#Mann= 3 , 0 , 0
       0      .1       0    60.1      .1       0   67.35      .1       0
Bank Sta=60.1,67.35
XS Rating Curve= 0 ,0
Exp/Cntr=0.3,0.1

Type RM Length L Ch R = 1 ,731.52  ,98.24,91.45,84.47
XS GIS Cut Line= 4
      637281.776    4315380.1781     637242.3265    4315355.8412
     637224.9622     4315321.673     637090.4819    4315327.7905
#Sta/Elev= 30
       0   809.9     2.9  808.91    5.79  807.57   23.18  803.22   46.35  794.32
   52.25  791.19    55.2  789.87   58.15  789.26   61.09  789.22   65.45  789.56
   75.83  791.02   84.68  791.78   87.74  792.66    90.8  793.08   93.86  793.21
   96.92  793.12  103.04  792.62   106.1  793.13  118.33  797.26  124.45  799.46
  127.51  800.82  130.57  801.42  139.75  801.95  151.99     803  161.17  803.34
  185.64  804.66  191.76  805.83  207.06   807.9  213.18  809.21   219.3  809.96
#Mann= 3 , 0 , 0
       0      .1       0    55.2      .1       0   65.45      .1       0
Bank Sta=55.2,65.45
XS Rating Curve= 0 ,0
Exp/Cntr=0.3,0.1

Type RM Length L Ch R = 1 ,640.0704,95.21,91.43,88.88
XS GIS Cut Line= 3
     637355.9918    4315274.8076     637283.3243    4315264.8694
     637128.9789    4315251.7888
#Sta/Elev= 30
       0  801.15    3.06  800.25    6.11  799.59   21.39  796.76   24.45  795.71
   39.73  791.46   42.78   790.8   45.84  789.06   55.01  786.32   58.06   785.7
   64.18     785   76.38  784.01   82.46  783.51   85.49  783.73   91.57  784.86
  106.75  787.38  121.94  788.25  124.98  788.65  131.05  789.99   143.2  792.95
  149.27  795.13  152.31  795.71   167.5   797.2  185.72  798.34  206.98  798.28
  210.02  798.39  213.06  798.68  216.09  799.17  225.21  800.86  228.24  801.99
#Mann= 3 , 0 , 0
       0      .1       0   76.38      .1       0   85.49      .1       0
Bank Sta=76.38,85.49
XS Rating Curve= 0 ,0
Exp/Cntr=0.3,0.1

Type RM Length L Ch R = 1 ,548.6401,88.11,91.44,94.97
XS GIS Cut Line= 3
     637363.9293    4315177.1761     637300.0662    4315162.4036
     637208.3261    4315198.2455
#Sta/Elev= 30
       0  791.93    5.96  791.37    14.9  790.16   17.88  789.35   20.86  788.03
    29.8  785.03   35.75  782.49   38.73  780.77   41.71  779.81   44.69  779.04
   47.67  778.47   50.65  778.25   56.61  778.23   65.55  778.41    74.5  779.15
   83.46  780.28   86.44  780.28   89.43  779.95   98.44  778.62  101.36  778.48
  104.35  778.68  107.33  779.62  110.32  780.21  125.24  782.75  128.23  783.62
  131.21  784.83  149.12  789.57   152.1  790.69  155.09  791.46  164.04  792.45
#Mann= 3 , 0 , 0
       0      .1       0   47.67      .1       0   65.55      .1       0
Bank Sta=47.67,65.55
XS Rating Curve= 0 ,0
Exp/Cntr=0.3,0.1

Type RM Length L Ch R = 1 ,457.2   ,119.54,91.44,54.83
XS GIS Cut Line= 6
     637393.2981    4315177.1761     637298.2008    4315099.6069
     637278.7721    4315089.6251     637261.2897    4315083.8645
     637243.1673    4315084.2611     637151.2039    4315181.1449
#Sta/Elev= 30
       0  792.14    6.14  789.57     9.2  788.84   12.27  788.99   15.34   787.9
   21.48  785.33   36.82  777.17   42.95  775.58    76.7  774.48   98.18  775.58
  119.65  775.29  144.56  775.72  147.63   775.2   150.7  774.13  153.77  773.91
   159.9  774.53  169.01  774.95  184.13  775.13  214.49  776.41  217.53  777.09
  220.56  778.39  232.71  784.48  238.78  786.99  253.96  788.14  260.03     788
  275.21  789.37  287.35  790.09   299.5  790.68  305.57  790.69  314.68  791.74
#Mann= 3 , 0 , 0
       0      .1       0   150.7      .1       0   159.9      .1       0
Bank Sta=150.7,159.9
XS Rating Curve= 0 ,0
Exp/Cntr=0.3,0.1

Type RM Length L Ch R = 1 ,365.76  ,102.85,91.44,75.79
XS GIS Cut Line= 6
     637414.8271    4315159.1824     637358.2115    4315039.8392
     637306.7764    4314984.8058     637270.9693    4315008.4857
     637242.0063    4315043.8609     637185.3889    4315118.8624
#Sta/Elev= 30
       0  782.31    6.14  777.02    9.22  775.27    21.5  774.27   36.86  773.88
    76.8  774.94   79.87  774.79   82.94  773.99   92.16  772.62  107.52  773.93
   119.8  773.32  138.12  771.87  165.24   770.8  186.33  770.54  207.42  770.77
  238.08  770.23  250.35  770.11  255.92  770.54  264.28  769.61  272.87  770.18
  293.18  771.15  302.15  772.78  308.21  773.19  332.46  773.97  353.68  773.99
  365.81  774.39  371.87  775.84  380.96  776.97  383.99  777.98  390.06  781.74
#Mann= 3 , 0 , 0
       0      .1       0  238.08      .1       0  272.87      .1       0
Bank Sta=238.08,272.87
XS Rating Curve= 0 ,0
Exp/Cntr=0.3,0.1

Type RM Length L Ch R = 1 ,274.32  ,90.94,91.44,88.76
XS GIS Cut Line= 6
     637419.3947    4315159.6394     637359.6142    4315038.8404
     637286.8272    4314961.7142      637209.357    4314943.5108
      637207.505    4314969.9692     637139.8003    4315111.2551
#Sta/Elev= 30
       0  782.82    3.06  780.73    6.13  777.82    9.19  775.69   12.25     775
   24.51  774.23   39.82  773.93   79.64  774.89   82.71  774.54   85.77  773.62
   88.83  773.57    91.9  772.77  110.28  774.03  140.84  771.78  165.08   770.9
  180.23  771.25  189.32  770.64  256.13  770.87  347.61  769.51  389.11  768.28
  396.62  767.76  400.16  768.18  406.64  770.07  429.89  771.21  480.87  771.85
  483.87  773.73  489.87  778.51  495.86  780.42  498.86  781.83  504.86  785.99
#Mann= 3 , 0 , 0
       0      .1       0  389.11      .1       0  400.16      .1       0
Bank Sta=389.11,400.16
XS Rating Curve= 0 ,0
Exp/Cntr=0.3,0.1

Type RM Length L Ch R = 1 ,182.8799,95.83,91.44,78.99
XS GIS Cut Line= 6
     637428.2768    4315164.7423     637360.8079    4315036.4191
     637287.3032    4314960.3513     637128.6356    4314919.6715
     637097.2824    4314987.9341     637061.4835    4315116.5467
#Sta/Elev= 30
       0  784.69    3.02   784.1    9.06  781.26    15.1  775.97   18.12  775.03
    30.2  774.38   48.33     774   87.59  774.87   99.67  772.81   117.8  774.06
     148  771.72  172.18  770.95  190.31  771.79   202.4  770.78  253.81  770.99
  308.67  770.13  378.28  769.73  408.55  768.54  443.44  766.41  455.25  765.78
  461.11  766.43  469.91  767.43  538.43  768.24  547.54  767.94  550.57  768.23
  574.84  771.28  596.08  778.79  602.15  780.62  611.25  781.01  623.39  782.68
#Mann= 3 , 0 , 0
       0      .1       0  443.44      .1       0  461.11      .1       0
Bank Sta=443.44,461.11
XS Rating Curve= 0 ,0
Exp/Cntr=0.3,0.1
