HEC-RAS study RedCreek.prj: RedCreek

--- RedCreek.g01 (geometry) --- (continued)

Type RM Length L Ch R = 1 ,10058.4 ,98.45,91.44,83.21
XS GIS Cut Line= 5
     637671.8785    4314775.2622     637655.0172    4315023.5429
     637634.9569     4315063.285     637624.3065    4315094.6704
     637614.1361     4315187.006
#Sta/Elev= 30
       0   799.4    6.14  797.49   21.51  793.69   24.58   793.6   33.79  791.36
   49.16  785.31    55.3  784.09   79.88  776.93   82.95  776.75    89.1  774.95
   92.17  774.79  122.89  776.97  141.32  778.25  159.76  778.88   199.7  779.34
  260.72  778.11  266.66  776.69  275.56  776.23   290.4  776.75  302.41  779.56
  308.44  779.46  314.46  777.71   341.5  778.94  389.44  779.11  392.44  779.39
  395.44  780.23  398.43  780.25  404.42  783.82  407.42  786.67  419.41  800.82
#Mann= 3 , 0 , 0
       0      .1       0   82.95      .1       0  122.89      .1       0
Bank Sta=82.95,122.89
XS Rating Curve= 0 ,0
Exp/Cntr=0.3,0.1

Type RM Length L Ch R = 1 ,9966.96 ,86.95,91.44,93.01
XS GIS Cut Line= 6
      637585.095    4314791.1372     637567.6988    4314990.6228
     637560.1291    4315007.9284     637554.4696    4315045.6563
     637542.8279    4315071.5855     637529.0032    4315193.3047
#Sta/Elev= 30
       0  800.91    18.2  796.44   21.24  796.41   33.37  793.39   54.61  789.99
   63.71  788.04   66.75  787.14   69.78   785.5   78.88  779.14   84.95  777.63
   91.02  774.92   97.09  773.34  115.29  775.04  136.53  776.29   169.9  775.87
  191.14  776.23  219.13  774.39  230.87  774.31  236.74  774.47  257.52  777.36
  277.41  775.17  285.94  776.13  368.63  779.01  371.69  779.53  374.75  781.72
  380.88  787.56  390.07  795.01  393.13  795.18  399.25  798.62  408.44  801.42
#Mann= 3 , 0 , 0
       0      .1       0   91.02      .1       0  115.29      .1       0
Bank Sta=91.02,115.29
XS Rating Curve= 0 ,0
Exp/Cntr=0.3,0.1

Type RM Length L Ch R = 1 ,9875.52 ,97.97,91.44,99.3
XS GIS Cut Line= 6
     637533.2366    4314766.7955     637492.3745    4314959.8626
     637470.3777    4314993.2842     637463.5348    4315001.6668
     637456.9202    4315065.9607     637493.0198    4315193.3047
#Sta/Elev= 30
       0  800.47   48.58  795.39   88.05  792.22  103.23  790.45  115.37  786.18
  118.41  786.19  121.44  784.86  127.51  780.88  130.55  778.34  133.59  776.51
  136.62  775.46   151.8  774.15  166.98  772.67  197.34  774.56   242.8  773.17
   245.5  773.38  248.21  774.44  254.08   776.2  271.71  776.09  283.46  774.77
  298.15  774.05  324.87  775.25  385.04  775.58   406.1  777.24   409.1  778.41
  418.13  786.15  433.17  796.58  436.18  796.73  439.19  798.59   445.2  800.81
#Mann= 3 , 0 , 0
       0      .1       0   151.8      .1       0  248.21      .1       0
Bank Sta=151.8,248.21
XS Rating Curve= 0 ,0
Exp/Cntr=0.3,0.1

Type RM Length L Ch R = 1 ,9784.08 ,89.96,91.44,97.66
XS GIS Cut Line= 6
     637495.1365    4314746.6872     637392.6499    4314944.6339
     637384.3449    4314967.9985     637362.1198    4315011.1257
     637380.3761    4315027.2653     637483.4948    4315193.3047
#Sta/Elev= 30
       0  801.38   33.59  797.98   79.39   794.5   88.55  792.65  125.19  782.49
  128.25  782.07  146.57  782.46  155.73  777.34  158.78  776.25     171  775.34
  180.16  772.78  186.26  771.46  219.85  772.11  227.06  772.91  232.76  774.72
  235.61  774.86  272.04  774.88   351.2  772.02  360.36  773.23   384.8  774.92
  433.66  774.73   464.2  775.82  470.31  777.69  473.36  779.64  476.42  779.67
  488.63  789.42  500.85  795.68   503.9  797.12  510.01  798.31  516.12  800.46
#Mann= 3 , 0 , 0
       0      .1       0  180.16      .1       0  227.06      .1       0
Bank Sta=180.16,227.06
XS Rating Curve= 0 ,0
Exp/Cntr=0.3,0.1

Type RM Length L Ch R = 1 ,9692.64 ,93.06,91.44,91.88
XS GIS Cut Line= 6
     637369.6973    4314787.9755     637314.2215    4314900.9071
     637282.2124    4314950.6811     637293.6424    4314953.2211
     637377.8198     4315027.802     637475.7425    4315193.3047
#Sta/Elev= 30
       0  801.04   24.55  796.07   36.83  794.49   70.58  788.56   92.06  783.72
  113.55  770.73  116.62  769.97  130.65  769.37  142.53  770.56  157.38  773.12
  166.29  771.91  177.15  771.31  233.23  771.53  248.42  773.04  263.62  773.75
  306.17  773.34  321.42  772.18  336.69  772.01  373.31     775  416.05  774.55
  449.63  775.45  452.68  776.05  458.78  779.55  461.83  779.75  464.89  781.39
  480.15  793.24   483.2  795.01  489.31  797.43  495.41  798.26  501.52  800.16
#Mann= 3 , 0 , 0
       0      .1       0  113.55      .1       0  233.23      .1       0
Bank Sta=113.55,233.23
XS Rating Curve= 0 ,0
Exp/Cntr=0.3,0.1

Type RM Length L Ch R = 1 ,9601.199,94.65,91.44,51.35
XS GIS Cut Line= 6
     637274.6587    4314761.5039     637222.1814    4314882.9098
     637192.1787    4314928.8233     637292.3854    4314954.2476
     637376.6799    4315029.9001     637471.5091    4315198.5964
#Sta/Elev= 30
       0  802.12   30.46     794    45.7  792.24   73.11  785.78   91.39  782.57
   94.44  781.57   97.48  778.96  103.58  770.65  106.62  768.09  117.74  767.63
  138.38  768.47  144.47  769.79  153.62  770.73  187.13   769.9  324.29  771.28
  357.97  773.57  388.58  772.71  397.76  773.14  419.24  771.88  431.53  772.21
  465.32  774.98   511.4  774.48  539.04  775.12  542.11  775.48  551.33   781.3
  557.47  783.08   575.9  797.28  582.05  799.02  588.19  799.17  597.41  801.55
#Mann= 3 , 0 , 0
       0      .1       0  103.58      .1       0  144.47      .1       0
Bank Sta=103.58,144.47
XS Rating Curve= 0 ,0
Exp/Cntr=0.3,0.1

Type RM Length L Ch R = 1 ,9509.76 ,100.44,91.44,118.05
XS GIS Cut Line= 6
     637156.1252    4314753.0372     637138.1702    4314846.7427
     637164.1927    4314923.4472     637291.2929    4314955.0486
     637373.8607    4315030.3998     637463.0425    4315194.3631
#Sta/Elev= 30
       0  801.16    5.96  800.45   29.82  794.06   35.78  793.28   56.65  787.08
   62.61  784.21   68.58     783   71.56   781.8   91.87  768.17   95.41  766.51
  104.26  766.03  119.02   766.6  124.92  768.07   156.6  770.09  204.91  769.83
  344.71  771.17  380.97  773.42  408.16  772.39  417.22   772.9   435.5  771.84
  484.46  774.97   527.3   774.4  554.84  774.94  560.95  775.92  570.13  782.18
  576.25  783.96  591.55  795.81  594.61  797.52  600.73  799.11  609.91  800.02
#Mann= 3 , 0 , 0
       0      .1       0   91.87      .1       0  124.92      .1       0
Bank Sta=91.87,124.92
XS Rating Curve= 0 ,0
Exp/Cntr=0.3,0.1

Type RM Length L Ch R = 1 ,9418.319,83.09,68.97,43.37
XS GIS Cut Line= 6
     637056.6416    4314773.1455     637048.0365    4314892.9491
      637231.314    4314943.5387     637290.2633    4314956.3446
     637369.7376    4315029.8416     637447.1674    4315175.8422
#Sta/Elev= 30
       0  792.64    9.09  789.86   18.18  784.16   27.27  779.61    30.3  779.55
   39.39  775.14   56.11  768.14   64.88  766.08   79.49     764   91.18   764.9
   97.02  766.33  102.29  767.78  135.52  766.65  166.18  766.92  187.65  767.36
  242.85   769.9  406.72  771.09  436.79   773.2  463.85  772.06  488.07  771.78
  518.67  773.89  527.85  773.43   540.1  774.91  576.82  774.24  610.49  774.92
  616.61  776.09  625.79  782.41  628.85  782.61  631.91  784.19  644.15  791.93
#Mann= 3 , 0 , 0
       0      .1       0   64.88      .1       0   97.02      .1       0
Bank Sta=64.88,97.02
XS Rating Curve= 0 ,0
Exp/Cntr=0.3,0.1

Type RM Length L Ch R = 1 ,9349.354,45.89,45.93,22.26
XS GIS Cut Line= 6
     636969.8581    4314763.0914     636983.7036    4314875.6016
     637230.9661    4314944.7198     637289.1745    4314957.4198
      637366.433    4315030.4449     637443.4632    4315176.9005
#Sta/Elev= 30
       0  792.13   17.81  777.34   20.78  776.52   23.74  774.97   35.62  765.09
   38.59  763.92   41.55  763.74   73.92  764.42  102.89  763.61  133.58  764.74
  155.19  766.69  204.28  766.53  244.17  767.13  304.97  769.83  421.05  771.01
  472.45  771.04  499.79  772.96  524.09  771.67   545.4   771.7  576.05  773.87
   588.3  773.03  603.63  774.95   640.4  774.12  671.04  774.92  674.11   775.3
   683.3  781.17  686.36  782.66  689.43  782.92  695.56  786.83  704.75  791.77
#Mann= 3 , 0 , 0
       0      .1       0   35.62      .1       0  133.58      .1       0
Bank Sta=35.62,133.58
XS Rating Curve= 0 ,0
Exp/Cntr=0.3,0.1

River Reach=Red Creek       ,2
Reach XY= 30
     636956.1954    4314870.4384     636709.0038    4314832.4949
     636624.0488    4314883.1089     636208.7135    4314981.6068
     635991.2591    4315065.4538     635847.6315    4315149.7013
     635724.1281    4315280.8512      635593.556      4315329.27
     635515.3714    4315305.0606     635174.0583    4315314.9825
     634893.4671    4315245.9261634842.2981571814315227.05852168
634813.4995924174315144.91014496634556.9120710074315079.97099456
634453.3299067794314989.76470295634398.6141642284314968.13569617
634202.9986355044314941.72644086633963.9709886454314947.97879893
633921.8351357724315024.67620295633827.8421929534315048.31475933
633739.3084073154315109.43825067       633640.18    4315144.3376
     633526.2299    4315143.5321     633315.8858    4315235.6073
      633282.683    4315226.9071     633252.7825    4315154.6447
     633201.9824    4315094.7164     633132.6345    4315128.3257
     632939.6475    4315151.4697     632755.1003    4315225.6854

Type RM Length L Ch R = 1 ,9303.427,42.48,32.85,32.33
XS GIS Cut Line= 4
     636929.9791    4314755.9753     636932.3604    4314848.8442
     636964.9042     4315105.226     636964.1104    4315212.3825
#Sta/Elev= 30
       0  789.32    8.99  785.21   20.98  774.24   29.97  764.59   32.96  763.03
   38.96  762.81   83.91  763.95  102.02  763.82  114.18  763.17  117.22  763.58
  120.26  764.76  129.38  766.26  132.43  766.24  214.52  763.69  260.12  764.45
  269.25  765.55  299.65  767.05  314.85   767.4  342.22  767.04  351.34  768.59
  360.52  771.63  363.59  771.95  369.71   774.9  375.83  777.09  391.14     779
  415.63     785  421.76  785.74  449.31   792.5  452.37  792.57   458.5  794.16
#Mann= 3 , 0 , 0
       0      .1       0   29.97      .1       0  120.26      .1       0
Bank Sta=29.97,120.26
XS Rating Curve= 0 ,0
Exp/Cntr=0.3,0.1

Type RM Length L Ch R = 1 ,9270.581,37.37,35.14,34.69
XS GIS Cut Line= 5
      636888.704     4314744.069     636889.4978    4314816.3004
     636900.6103    4314860.7505     636926.0104    4315044.9009
     636918.0728    4315283.0264
#Sta/Elev= 30
       0  791.67    3.01  789.92    9.03  787.77   21.07  778.17   27.09  775.69
   33.11  770.35   39.13  763.93   42.14  762.59   51.17  763.04   127.2  762.58
  133.29  763.06  139.39  764.74  148.53  765.64  227.76  763.48  264.33   763.2
  267.38  763.73  273.47  766.25  276.52  766.69  368.09  766.89  386.42  767.62
  389.48  768.66  401.69  776.13  413.91  777.67   441.4   783.1  465.84  788.65
  471.95  789.43  499.44  797.05   502.5  797.16  520.82  801.14  542.21  803.83
#Mann= 3 , 0 , 0
       0      .1       0   39.13      .1       0  267.38      .1       0
Bank Sta=39.13,267.38
XS Rating Curve= 0 ,0
Exp/Cntr=0.3,0.1

Type RM Length L Ch R = 1 ,9235.439,40.93,91.44,116.87
XS GIS Cut Line= 6
     636853.1568     4314726.054     636851.7265    4314826.0173
     636860.5298    4314840.0014     636871.8349    4314918.0925
     636878.3828     4314938.937     636867.4443    4315326.1302
#Sta/Elev= 30
       0  800.18    6.06  796.94   15.15  790.48   21.21  789.02   30.29  785.02
   42.41  775.83   48.47   774.2   54.53  771.03   63.62  762.67   66.65  761.99
   116.5  762.74  142.48  762.21  168.65   764.9  272.65  762.33  275.73  762.47
   278.8  763.94  281.88  765.47  284.95   765.8  309.54  765.34  340.29  765.84
  380.25  764.79  407.92  766.25  417.14  767.98  426.36  772.78  435.59  775.69
   469.4  779.43  521.66  788.17  558.55  792.71  583.15  798.17  604.67  800.15
#Mann= 3 , 0 , 0
       0      .1       0   63.62      .1       0   278.8      .1       0
Bank Sta=63.62,278.8
XS Rating Curve= 0 ,0
Exp/Cntr=0.3,0.1

Type RM Length L Ch R = 1 ,9144    ,143.38,91.44,43.25
XS GIS Cut Line= 5
     636835.6943     4314722.879     636831.2824    4314805.0429
     636770.8681    4314890.4726     636754.4655    4314962.3309
      636721.394    4315375.3428
#Sta/Elev= 30
       0  800.26    6.09  797.84   18.28  789.01   30.47  785.33   39.62  783.63
   48.76  779.67   54.85  777.98   60.95  774.23      64  771.08   70.09  762.73
   73.14  761.57  151.04  761.26  160.01  760.63  165.99  760.72  180.94  763.13
  236.05  759.68  254.48  761.69  282.11  760.07  285.18  760.63  288.24  762.27
  291.31  763.14  328.14  762.44  417.15  763.44  432.49  768.09  463.19  772.01
  509.22   775.7  533.78   779.8  570.61  783.64   601.3  787.79  674.96  800.53
#Mann= 3 , 0 , 0
       0      .1       0   70.09      .1       0  288.24      .1       0
Bank Sta=70.09,288.24
XS Rating Curve= 0 ,0
Exp/Cntr=0.3,0.1

Type RM Length L Ch R = 1 ,9052.56 ,92.84,91.44,66.62
XS GIS Cut Line= 6
     636654.7189    4314737.1665     636682.6126     4314816.788
     636699.5764    4314828.2487       636733.36    4314885.2746
     636703.3732    4314967.6623     636669.0064    4315335.6552
#Sta/Elev= 30
       0  792.86    3.01  791.41    9.04  790.02   21.09  784.55   30.13  781.68
   42.18  780.62   66.29  776.47   75.33  772.69   84.37  771.35   87.29  770.47
   98.99  763.68  104.84  762.42  107.69  760.75  113.39  759.64  139.03  759.91
  147.81   760.2  168.29  762.52  222.62  759.04  252.85  759.14   258.9  760.45
     265  761.73  341.37  762.69   365.8  762.22   399.4  763.37  402.46  763.83
  411.62  767.65  414.67  768.23  588.78   786.2  604.05  787.95  628.49  792.52
#Mann= 3 , 0 , 0
       0      .1       0  107.69      .1       0   258.9      .1       0
Bank Sta=107.69,258.9
XS Rating Curve= 0 ,0
Exp/Cntr=0.3,0.1

Type RM Length L Ch R = 1 ,8961.12 ,82.11,91.7,52.83
XS GIS Cut Line= 4
     636573.7562    4314767.3291     636622.2935    4314872.0454
      636665.355    4314944.5822     636629.3189    4315270.5676
#Sta/Elev= 30
       0  784.61   15.19  781.32   45.56  776.89   51.63  776.42   75.93     772
   88.08  770.76   94.16  768.47  106.31  762.47  112.38  760.78  115.42  759.26
  118.43  758.12  121.44  757.71  130.48  757.92  139.52  760.03  145.55  760.51
  169.65  758.27  178.68  757.99  196.76  758.67  202.84  759.41   224.3  760.86
  319.31  761.49   346.9  762.32  349.97  762.92   356.1  765.37  371.42  768.94
  405.14   771.2   417.4  773.05  512.42   780.6  521.61  781.92  527.74  783.66
#Mann= 3 , 0 , 0
       0      .1       0  115.42      .1       0  202.84      .1       0
Bank Sta=115.42,202.84
XS Rating Curve= 0 ,0
Exp/Cntr=0.3,0.1

Type RM Length L Ch R = 1 ,8869.417,51.17,50.31,121.68
XS GIS Cut Line= 6
     636511.8436    4314772.0916     636552.8636    4314934.4232
     636628.0054    4314937.8628     636621.6554    4314955.8545
     636622.7137    4314972.7879     636594.3938    4315264.2176
#Sta/Elev= 30
       0  784.14     9.1  781.05   18.19  779.09   87.93  770.68   90.96  769.89
  106.12  762.77  112.18  761.71  124.31  757.94  130.37  756.25  139.47  755.66
  145.53   755.9  151.02  757.91  156.52  758.62   167.5  757.85  182.54  758.34
  242.72   757.5  248.17  758.08  253.62  759.41  259.07  759.64  297.06  759.47
  351.96  760.55  364.16  760.29  385.51  762.34  397.71  765.58  412.96  767.47
  461.76  772.31  525.81  777.45  544.11  778.03  565.46  782.04  571.56  782.49
#Mann= 3 , 0 , 0
       0      .1       0  124.31      .1       0  248.17      .1       0
Bank Sta=124.31,248.17
XS Rating Curve= 0 ,0
Exp/Cntr=0.3,0.1

Type RM Length L Ch R = 1 ,8819.107,43.62,40.87,37.78
XS GIS Cut Line= 5
     636451.7438    4314784.3916     636501.7501    4314933.6169
     636500.9564    4314955.0482     636502.5439    4314993.1483
     636532.7065    4315242.3863
#Sta/Elev= 30
       0  782.13   15.13   778.2   66.58  773.69   78.69  771.71   87.77  770.95
    90.8  769.91   99.88  765.16  105.93  762.64  111.98  761.46  122.08  757.23
  127.12  755.45  130.14  755.27  163.51  755.58  169.64  756.91  175.76  758.85
  178.83  759.08  262.89   758.3     318  757.05  321.06  757.54  339.43  765.86
  345.55  767.29  354.74  768.04  363.92  767.98  382.29  769.52  403.72  772.94
  406.78  772.95  431.28  777.75  440.46  778.47  461.89  781.52  468.02  781.96
#Mann= 3 , 0 , 0
       0      .1       0  122.08      .1       0  169.64      .1       0
Bank Sta=122.08,169.64
XS Rating Curve= 0 ,0
Exp/Cntr=0.3,0.1

Type RM Length L Ch R = 1 ,8778.239,90.64,91.44,90.72
XS GIS Cut Line= 6
     636393.7334    4314792.5175     636449.4554    4314913.2389
     636452.7292    4314916.4298      636463.316    4314938.7176
     636462.6052    4314955.8986     636491.1002    4315231.7267
#Sta/Elev= 30
       0  783.23   54.39  773.85   63.46  771.42    69.5  768.99   84.61   768.8
   90.66  767.12   99.72  762.47  105.76  760.29   123.9  757.76  129.94   755.8
  135.25  755.04  162.21  754.94  165.07  755.18  167.94  756.33   170.8  757.59
  176.54  758.11  200.73  757.28  264.72  757.56  331.76  756.21  334.81  757.09
   340.9  760.54  350.05  764.88  359.19  766.23  368.33  768.46  380.52   770.6
  386.61  771.14  407.94  774.91  414.04  775.55  438.42  780.44   456.7  782.88
#Mann= 3 , 0 , 0
       0      .1       0  129.94      .1       0  167.94      .1       0
Bank Sta=129.94,167.94
XS Rating Curve= 0 ,0
Exp/Cntr=0.3,0.1

Type RM Length L Ch R = 1 ,8686.8  ,98.31,91.44,79.48
XS GIS Cut Line= 4
     636360.0783    4314795.3397     636366.1107    4314941.5153
     636370.7014    4314974.3846     636470.1452    4315225.0239
#Sta/Elev= 30
       0  783.08    3.05  782.96   18.29  780.27   24.38  779.75   36.58  777.79
    76.2  773.18   82.29  772.79   85.34  772.07  100.58  766.75  109.73  760.41
  112.77  760.17  118.87  754.55  121.92  754.05  143.25  754.39  155.35  753.59
   164.4   754.8  240.77  756.93  280.61  755.59  338.82  756.14  341.89  757.46
  348.02  762.15  360.27  765.33   366.4   767.7  372.53  769.44  378.66  770.71
  390.92  772.14  412.37   775.9  415.43  775.94  439.94  780.81  449.14  782.07
#Mann= 3 , 0 , 0
       0      .1       0  118.87      .1       0   164.4      .1       0
Bank Sta=118.87,164.4
XS Rating Curve= 0 ,0
Exp/Cntr=0.3,0.1

Type RM Length L Ch R = 1 ,8595.359,93.7,91.46,96.47
XS GIS Cut Line= 6
     636197.0947    4314799.5731     636275.6332    4314958.8056
     636279.7891    4314970.8956     636297.2772    4315009.4533
     636317.4184    4315047.7785     636385.4784     4315263.124
#Sta/Elev= 30
       0  782.51    9.18  780.49   15.31  779.81   24.49  777.93   64.28  773.04
   91.84  771.12  122.45  769.69  134.69  766.36  137.75  766.27     150  762.49
  153.06   761.1   165.3  753.64  168.36  753.45  171.43  752.62  185.22  752.37
   199.4  753.39  217.55  754.82  255.76  756.18   330.9  754.57  352.26  754.63
  364.47   755.2  367.52  755.97  379.73  762.44  382.78  762.98  388.89  765.04
   401.1  767.64   413.3  769.03  434.67  773.41  456.03  775.13  501.81  782.18
#Mann= 3 , 0 , 0
       0      .1       0  168.36      .1       0   199.4      .1       0
Bank Sta=168.36,199.4
XS Rating Curve= 0 ,0
Exp/Cntr=0.3,0.1

Type RM Length L Ch R = 1 ,8503.904,101.55,91.42,91.47
XS GIS Cut Line= 4
     636110.3112    4314791.1064     636167.6639    4314957.9522
     636188.6781    4314983.8064     636298.6949    4315280.0574
#Sta/Elev= 30
       0  783.42    6.08  782.93   30.42  778.46    36.5  777.91   60.84  773.86
   91.26  770.94  155.13  767.61  182.49  761.18  188.54  760.27  200.66  753.14
  203.69  751.85  206.72  751.32  228.15  751.19   243.5  752.08  289.52  754.73
  332.47  753.77  344.74  753.02  353.95  753.54  378.49  753.01   387.7  752.55
  393.83  751.54  399.97  753.88  406.11  759.77  409.17  761.75  412.24  762.66
  449.06  767.79  467.47  769.26  473.61  771.74  495.08  774.06  525.76  781.83
#Mann= 3 , 0 , 0
       0      .1       0  203.69      .1       0   243.5      .1       0
Bank Sta=203.69,243.5
XS Rating Curve= 0 ,0
Exp/Cntr=0.3,0.1

Type RM Length L Ch R = 1 ,8412.479,90.61,91.42,85.47
XS GIS Cut Line= 6
     635907.1107    4314532.8725     636093.1835    4315005.2687
     636101.0304    4315010.9642     636107.1317    4315026.5217
     636109.3232    4315036.7541     636208.7364    4315287.3334
#Sta/Elev= 30
       0  783.12   21.41  779.52    36.7  777.92   85.64   776.8  128.46   774.1
  143.75     772  155.99  771.94   177.4  773.76   214.1  773.99  238.57  777.65
  278.33   777.3  311.97  779.05  330.32  778.78  385.38  773.15   428.2  770.76
   464.9  766.96  495.49  760.08  498.55  758.31  507.72   750.7  522.99  749.35
  539.36  750.44  572.17  752.51   602.8  752.78  734.53  749.51  737.59  750.35
  752.91  759.86  765.16  765.76  780.48   770.7  798.86   775.3  814.18  782.97
#Mann= 3 , 0 , 0
       0      .1       0  507.72      .1       0  539.36      .1       0
Bank Sta=507.72,539.36
XS Rating Curve= 0 ,0
Exp/Cntr=0.3,0.1

Type RM Length L Ch R = 1 ,8321.056,96.45,91.46,86.83
XS GIS Cut Line= 3
     635864.2482    4314692.0197     636023.6525    4315061.8421
     636131.7413    4315301.7553
#Sta/Elev= 30
       0  782.79   30.74  779.74   49.19  773.95   73.78  769.25   92.22  767.85
  110.67  763.43     166  766.46   190.6  765.46  199.82  763.89  288.97  765.65
  295.12  764.68  316.64  765.46  341.23  763.52  359.68  760.07  371.97  749.89
  421.07  749.77  460.85  751.43  503.69   750.7  531.22  751.81   540.4  750.59
   555.7   750.8  567.94  748.73  604.66   750.4  619.96  748.52  623.02  749.14
  632.19  757.84  635.25  759.14  641.37  766.23  656.67  780.58  665.85  782.63
#Mann= 3 , 0 , 0
       0      .1       0  371.97      .1       0  421.07      .1       0
Bank Sta=371.97,421.07
XS Rating Curve= 0 ,0
Exp/Cntr=0.3,0.1

Type RM Length L Ch R = 1 ,8229.6  ,86.31,91.44,98.15
XS GIS Cut Line= 6
     635678.5103    4314733.2948     635924.8751    4315074.3431
     635930.5009    4315083.6314     635947.1722     4315107.336
     635961.0327       4315135.8     636047.5802    4315318.7094
#Sta/Elev= 30
       0  782.31   42.99  782.13   76.77  780.78  138.19  775.53  171.98  773.45
  208.83  772.43  242.61   769.9  267.18  763.55  331.67  759.02  340.88  757.55
  356.23   752.1  383.87  753.18  408.44  751.98  414.58  750.84  420.72  748.22
  426.15  748.01  437.38  747.25  492.22  748.07  565.81  750.07  578.07  748.46
  611.79   749.3  642.45  748.01  645.52   748.4  648.59  750.31  654.72   755.7
  657.78  755.97  660.85  757.76  685.38  776.52  688.44  776.83  694.58   781.5
#Mann= 3 , 0 , 0
       0      .1       0  426.15      .1       0  492.22      .1       0
Bank Sta=426.15,492.22
XS Rating Curve= 0 ,0
Exp/Cntr=0.3,0.1

Type RM Length L Ch R = 1 ,8138.16 ,101.26,91.44,75.94
XS GIS Cut Line= 5
     635659.4603    4314774.5699     635861.2108    4315135.8761
     635864.9822    4315150.8595     635870.9287    4315160.4328
     635932.5108     4315342.896
#Sta/Elev= 30
       0  781.94   18.39  778.01   33.72  777.12   58.24  774.22   73.57  773.57
   98.09  773.86  116.48  773.48  153.27  771.02  202.31  768.49  288.14  766.07
  327.99  758.31  361.71  755.16  373.97  753.35  398.49  751.77  401.56  750.58
  404.62  748.16  407.69  746.53  413.82  745.38  424.12  744.92  452.77  746.35
  486.39  748.18  544.47  746.55  578.09   746.4  587.26  748.84  593.38  749.68
  596.43  751.13  617.83   769.6  620.89  770.97  623.94  773.12  633.11  780.79
#Mann= 3 , 0 , 0
       0      .1       0  407.69      .1       0  452.77      .1       0
Bank Sta=407.69,452.77
XS Rating Curve= 0 ,0
Exp/Cntr=0.3,0.1

Type RM Length L Ch R = 1 ,8046.72 ,96.26,91.44,78.61
XS GIS Cut Line= 6
     635628.2063    4314877.6584     635761.5249    4315160.2578
     635788.8033    4315196.4455     635803.0345    4315209.4645
     635801.7116     4315217.402     635890.4819    4315344.6355
#Sta/Elev= 30
       0  772.41    3.06  771.22    6.13  770.81   64.33  770.79  110.28  766.95
  177.68  765.09  248.14  762.31  275.71  760.15  300.21  756.83  306.34  755.56
  321.53   751.1  327.57  749.83   345.7  749.49  348.72     749  357.79   745.6
   360.5  745.06  365.93  744.79  385.32  744.11  409.65  744.87  443.11   745.7
  461.37  744.91  467.45  744.99  497.87  746.17     507  746.85  510.04  747.71
  513.08  749.86  528.29  762.85  531.33  764.04  534.37  766.19  540.46  771.35
#Mann= 3 , 0 , 0
       0      .1       0  365.93      .1       0  409.65      .1       0
Bank Sta=365.93,409.65
XS Rating Curve= 0 ,0
Exp/Cntr=0.3,0.1

Type RM Length L Ch R = 1 ,7955.28 ,84.2,91.44,106.89
XS GIS Cut Line= 6
     635618.6813    4314887.1834     635698.3727    4315218.7759
     635726.6883    4315264.5509      635756.177    4315290.7024
     635775.2532    4315311.9466     635806.0066    4315366.6094
#Sta/Elev= 30
       0  771.27    3.07  770.55    6.14  770.43    55.3  770.38   70.66  769.96
  129.04  765.67  168.98  764.18  193.56  762.58  215.07  760.29  221.21  760.12
  251.94  757.94  276.51   755.3  291.88  754.47  310.31  751.28   322.6  747.08
  325.67  746.33  367.95  744.25  388.88  743.15  445.69  742.75  465.81   742.3
  471.79  742.68  483.73   744.1  489.71  744.92  492.69  746.33  495.68  748.89
  501.65  755.03  504.64  757.69  507.63  758.31  510.61  760.69  525.55  774.51
#Mann= 3 , 0 , 0
       0      .1       0  367.95      .1       0  483.73      .1       0
Bank Sta=367.95,483.73
XS Rating Curve= 0 ,0
Exp/Cntr=0.3,0.1

Type RM Length L Ch R = 1 ,7863.84 ,85.72,91.44,104.43
XS GIS Cut Line= 5
     635601.2187    4314844.3208     635640.3127     4315280.372
     635665.1126    4315331.6268      635668.959    4315341.6461
     635672.6564    4315395.1844
#Sta/Elev= 30
       0  783.28   21.43  778.99   30.62  777.63   36.74   776.1   55.11  770.31
   61.23  769.73  134.71  768.33  153.08  767.48  208.18  763.82  232.68   761.7
  266.35  759.49   278.6  758.29  290.85  756.12  300.03   755.8  327.58   753.2
  330.65   752.3  342.89  747.11  352.08  745.51   358.2  745.07  425.55  743.65
  494.74  742.26  497.42  742.26  505.47  743.54  511.43  749.66  526.34     762
   532.3  766.35  535.29  766.75  538.27  768.52  547.21  775.64  559.14  785.86
#Mann= 3 , 0 , 0
       0      .1       0  425.55      .1       0  505.47      .1       0
Bank Sta=425.55,505.47
XS Rating Curve= 0 ,0
Exp/Cntr=0.3,0.1

Type RM Length L Ch R = 1 ,7772.4  ,99.27,91.44,91.04
XS GIS Cut Line= 6
     635593.2812    4314850.6708     635572.1498    4315306.3959
     635567.5383    4315316.4979     635565.0662    4315330.3779
      635565.006    4315337.8284     635563.1187    4315474.5596
#Sta/Elev= 30
       0  783.25   18.37  779.27   24.49  778.44   48.99  771.09    64.3  768.16
  131.66  767.64  208.21  762.52  257.19  757.89  266.38  757.62  290.88  753.51
  293.94  753.45     297  752.57  312.31  745.75  318.43  744.19  342.93  743.14
  410.29  742.92  481.42  741.67  486.39  742.54  497.99  752.36  504.06  756.85
   507.1  757.23  519.26   762.8  534.45  766.33  543.57  767.56  564.84  772.75
  576.99  773.55  583.07  772.46  598.27  773.73  610.42  776.33  625.61  780.86
#Mann= 3 , 0 , 0
       0      .1       0  410.29      .1       0  486.39      .1       0
Bank Sta=410.29,486.39
XS Rating Curve= 0 ,0
Exp/Cntr=0.3,0.1

Type RM Length L Ch R = 1 ,7680.96 ,103.64,91.44,87.96
XS GIS Cut Line= 5
     635593.2812    4314803.0457     635483.0817    4315286.0142
     635480.2436    4315315.0263     635477.8565    4315318.7299
     635459.9309    4315384.0719
#Sta/Elev= 30
       0  790.91    9.17  789.07   12.23  789.03   45.87  783.82   70.33  777.56
   76.45  776.68  103.97  768.54  113.14     767  146.78  766.63  204.88  764.46
   269.1  761.35   290.5  759.24  296.62  759.17  299.67  758.27  311.91  750.83
  324.14  746.29  339.43  743.53  452.57  741.85  524.53  740.01  526.73  740.07
  528.94  741.08  537.78  750.22  546.61  757.73  549.56   759.8  552.51   759.9
  573.13  775.13  579.02   780.3  581.96  782.02  584.91  782.59  596.69  790.78
#Mann= 3 , 0 , 0
       0      .1       0  452.57      .1       0  528.94      .1       0
Bank Sta=452.57,528.94
XS Rating Curve= 0 ,0
Exp/Cntr=0.3,0.1

Type RM Length L Ch R = 1 ,7589.52 ,95.19,91.44,86.7
XS GIS Cut Line= 6
      635478.981    4314672.8705     635379.6628    4315214.1972
     635386.7816    4315275.7149     635389.4995    4315310.6285
     635388.6587    4315320.3482     635393.2558    4315392.0094
#Sta/Elev= 30
       0   792.6   27.52  788.14   73.38  783.46   82.55  781.76  107.01  773.06
  119.25  766.44  125.36  763.99  165.11  760.54  177.34   757.2  189.57  759.38
  210.97   761.5  232.38  760.65  256.84  757.61   302.7  755.17  373.02  755.26
     425  748.21  446.41  742.29  461.69  742.04  473.92  740.74  553.31  740.08
  641.47  738.45  652.19  739.93  657.07  743.45  660.06  744.01  672.03  756.24
  686.99  769.59  689.98  769.82  713.91  786.24  722.89  790.14  728.87  794.18
#Mann= 3 , 0 , 0
       0      .1       0  553.31      .1       0  652.19      .1       0
Bank Sta=553.31,652.19
XS Rating Curve= 0 ,0
Exp/Cntr=0.3,0.1

Type RM Length L Ch R = 1 ,7498.08 ,88.26,91.44,98.24
XS GIS Cut Line= 4
     635421.8309    4314650.6454      635292.944    4315275.2199
     635305.8349    4315324.0406     635263.7156    4315441.9628
#Sta/Elev= 30
       0  783.48   12.26  781.61   27.59  776.66   42.92  776.03   70.52  771.56
   95.05  769.49  107.31  767.19  122.64  762.27  156.37  760.11  174.76  756.31
  229.95  757.14  309.67  751.94  407.78  753.26  423.11  751.86  444.57  746.08
  456.84  744.85   469.1  740.83   496.7  739.52  588.68  739.72   640.7  737.93
  685.26  736.39  691.28  738.66  697.39  743.97   703.5  747.13  730.99  770.72
   743.2  776.26  770.69  773.07  792.07  772.11  801.23  773.74  813.45  784.62
#Mann= 3 , 0 , 0
       0      .1       0   640.7      .1       0  691.28      .1       0
Bank Sta=640.7,691.28
XS Rating Curve= 0 ,0
Exp/Cntr=0.3,0.1

Type RM Length L Ch R = 1 ,7406.64 ,95.44,91.44,93.71
XS GIS Cut Line= 6
     635349.0086    4314693.5609      635212.975    4315300.5045
     635212.1797    4315309.9111     635211.0215    4315314.9487
     635209.9322    4315332.1419     635199.1328    4315379.9356
#Sta/Elev= 30
       0  781.44    9.19  780.51   24.51  777.62   36.77  774.59   39.83   774.7
   55.15  770.78   73.54  767.89   88.86  764.57  107.24  761.99  125.63   757.7
  140.95  756.84  180.78  753.13  248.19     751  337.05  751.72  358.49  750.37
  361.56  749.76  379.94  741.86   392.2  741.32  413.65  739.18  447.35  738.04
  585.23  737.68  629.08  735.78  645.35  735.66  651.01  736.17  653.84  738.07
  669.15   754.2  672.22  754.52  696.72  779.42  699.78  782.16  702.84   783.3
#Mann= 3 , 0 , 0
       0      .1       0  585.23      .1       0  653.84      .1       0
Bank Sta=585.23,653.84
XS Rating Curve= 0 ,0
Exp/Cntr=0.3,0.1

Type RM Length L Ch R = 1 ,7315.2  ,102.42,91.44,96.88
XS GIS Cut Line= 6
     635258.0027    4314765.6049     635130.3543    4315286.2324
     635123.1914    4315296.7496      635119.246    4315307.3613
     635118.0776    4315315.0191     635107.6007    4315353.5526
#Sta/Elev= 30
       0  772.46    6.13  770.59   42.88  763.21   55.14   759.7   70.45  757.77
  131.71  751.71  165.41  749.19   174.6  748.84  180.72  750.29  186.85  750.45
  238.92  747.44  275.68  739.08   349.2  739.71  361.45  738.78  367.58  736.89
  382.89   736.1  416.59  737.28  447.22  736.16   465.6  735.52  514.61  737.17
  529.92  736.95  541.14  735.66  562.68  736.26  567.84  737.48  570.91  739.22
  573.98  741.85   583.2  752.02  586.27  754.58  589.34  755.37  607.77  774.38
#Mann= 3 , 0 , 0
       0      .1       0  447.22      .1       0  562.68      .1       0
Bank Sta=447.22,562.68
XS Rating Curve= 0 ,0
Exp/Cntr=0.3,0.1

Type RM Length L Ch R = 1 ,7223.76 ,93.78,91.44,75.23
XS GIS Cut Line= 6
     635191.8568    4314717.8475     635044.7476    4315245.3459
     635037.7837    4315262.9802     635034.0416    4315274.1413
     635029.3624      4315280.35     635003.7377    4315346.1019
#Sta/Elev= 30
       0  783.28    9.18  781.15   27.53  774.71   48.95  773.51   67.31  769.19
    82.6  767.87  100.96  761.39   113.2  758.56  192.74  750.83  204.98  750.47
  244.75  744.97  260.05  745.77  296.76  741.41  327.35  738.98  357.95  737.22
  419.13  735.68  440.55  733.87   489.5  735.18   504.8   734.3  541.51  734.61
  553.04  736.83  561.17  737.46  576.14  734.57  598.41  733.66  601.48  734.11
  604.55  736.08  622.96  753.42  626.03  755.54   629.1  756.26  656.71  782.56
#Mann= 3 , 0 , 0
       0      .1       0   489.5      .1       0  601.48      .1       0
Bank Sta=489.5,601.48
XS Rating Curve= 0 ,0
Exp/Cntr=0.3,0.1

Type RM Length L Ch R = 1 ,7132.32 ,92.89,91.44,97.29
XS GIS Cut Line= 6
     635102.4274    4314563.3967     634947.4731    4315243.9721
     634943.2919    4315264.5144     634948.6326    4315270.2394
     634954.7709    4315286.1144         634945.    4315338.6274
#Sta/Elev= 30
       0  780.95   12.25  781.93   67.35  776.04   91.84  777.11  122.45  774.38
  165.31  766.85  186.74  764.95  211.23  758.45  220.42  757.11  238.79  757.69
  254.09  756.35  263.28  757.14  303.08  752.89  394.92  747.83  419.41  743.81
  446.96     736  526.55  733.44   578.6  734.01  609.21  733.14  630.64  732.32
  667.38  732.87  691.87   736.6  712.97   732.6   735.3  733.15  738.13     735
  752.71     750  755.68  750.41  782.38  774.36  788.32  776.92  797.22  784.56
#Mann= 3 , 0 , 0
       0      .1       0  609.21      .1       0   735.3      .1       0
Bank Sta=609.21,735.3
XS Rating Curve= 0 ,0
Exp/Cntr=0.3,0.1

Type RM Length L Ch R = 1 ,7040.88 ,90.96,91.47,96.08
XS GIS Cut Line= 6
     634988.6564    4314675.8448     634863.5635    4315191.7617
     634857.3039     4315229.333     634856.6196    4315232.3123
     634860.7678    4315246.4163     634847.3951    4315309.1528
#Sta/Elev= 30
       0  783.12   24.55  780.21    49.1  775.35   52.17  775.29   67.51  770.59
   76.71  766.78   85.92  765.57  110.47  757.21  171.84  751.19  291.52  744.57
  309.93     742  319.13  739.79  325.27  737.66  331.41  733.88  334.48  733.39
  346.75     734  383.57  733.91  463.36  731.67  509.39  731.17   554.3  733.47
  563.09  732.01  572.01  730.79  583.77  732.07  586.71  732.79  589.77  734.66
  592.82  734.95  620.31  759.76  623.37  760.31  626.42  762.49  650.86  783.15
#Mann= 3 , 0 , 0
       0      .1       0  563.09      .1       0  583.77      .1       0
Bank Sta=563.09,583.77
XS Rating Curve= 0 ,0
Exp/Cntr=0.3,0.1

Type RM Length L Ch R = 1 ,6949.409,94.32,91.41,90.28
XS GIS Cut Line= 4
     634928.0931    4314662.2452     634780.9009    4315195.6865
     634770.2163    4315219.7992     634746.8532    4315294.6006
#Sta/Elev= 30
       0  782.76   27.52  779.22   55.03  773.23    64.2  771.93   79.49  767.89
  107.01  755.84  119.24  753.48  143.69  752.38  162.04  749.46  180.38  747.98
  189.55  745.79  244.59  744.36  284.33  741.89  305.73   737.4   314.9  733.58
  317.96  733.07  412.74  733.15  467.77  730.81  489.17  729.63  550.32  732.95
   565.1  732.01  570.96  730.66  585.78  731.29  588.79  731.63  594.82  734.77
  597.84  735.34  618.93  756.75  624.96  762.04  630.99  764.16  658.12  783.65
#Mann= 3 , 0 , 0
       0      .1       0  467.77      .1       0  585.78      .1       0
Bank Sta=467.77,585.78
XS Rating Curve= 0 ,0
Exp/Cntr=0.3,0.1

Type RM Length L Ch R = 1 ,6858    ,96.66,91.44,94
XS GIS Cut Line= 6
     634876.4993    4314573.6096     634693.9851    4315165.8491
     634686.4155    4315184.1241     634677.4751    4315212.4159
     634675.9934    4315227.2326     634662.1863    4315273.4339
#Sta/Elev= 30
       0  782.49   27.61  779.68   39.88   781.5  104.31  776.24  131.92  771.56
  147.26  765.71  150.33  765.37  174.87  755.61  181.01  753.71  196.35  751.09
  245.44  745.51  282.25  742.85  303.73  739.96  365.09  735.46  380.43  731.15
  500.08  730.16  518.48  731.55  530.76  730.24  536.89  729.18   555.3  728.52
  616.66  729.99  663.82  731.43  666.51  732.99  675.16   742.8  678.14   742.9
  693.14  759.26  699.16  764.58  705.19  768.74  711.22  770.67  732.32   783.4
#Mann= 3 , 0 , 0
       0      .1       0  530.76      .1       0  616.66      .1       0
Bank Sta=530.76,616.66
XS Rating Curve= 0 ,0
Exp/Cntr=0.3,0.1

Type RM Length L Ch R = 1 ,6766.56 ,92.96,91.44,88.47
XS GIS Cut Line= 5
     634781.2491    4314627.8493     634596.8892    4315164.8534
      634594.313    4315174.2829     634589.4084    4315183.4087
     634572.5586    4315235.5323
#Sta/Elev= 30
       0  783.74   12.28  782.08    39.9  774.99   42.97  774.89   70.59  763.41
   76.73  762.13   92.07  755.68  107.42  751.83  110.48  751.77  125.83  748.66
  193.35  741.81   257.8  737.18   297.7  732.98  340.66  731.65  349.87  730.64
  359.08   730.8  371.35  729.06  423.53  731.15  454.22  728.54  472.63  727.61
  561.63  727.85  572.66  728.39  582.73  728.96  585.32  730.09  587.91   732.7
  603.12  751.25  609.21  755.41  621.38  767.79  639.64  782.47  642.68   783.5
#Mann= 3 , 0 , 0
       0      .1       0  454.22      .1       0  572.66      .1       0
Bank Sta=454.22,572.66
XS Rating Curve= 0 ,0
Exp/Cntr=0.3,0.1

Type RM Length L Ch R = 1 ,6675.12 ,109.74,91.44,88.49
XS GIS Cut Line= 6
     634650.7431    4314639.4249     634522.4598    4315107.8612
     634512.2532     4315130.206     634507.5337    4315145.0486
     634506.8494    4315152.3113     634490.6248    4315196.6237
#Sta/Elev= 30
       0  773.26    12.3  767.81   18.44  766.06   33.81  758.95   49.18  756.23
   76.85  749.21  126.03   741.2  165.99  740.02  242.84  733.48  248.99  731.87
  258.21  731.68  267.43  732.34  301.25  728.31  313.54  728.96  356.58   729.3
  393.47  728.89  421.13  727.76  442.65  726.25  451.87  728.52  464.17   726.6
  501.04  726.05  512.84  726.15  528.26   727.3  530.69  728.29  539.02  733.56
  553.76   753.6  559.66  759.29  565.56  763.92  571.46  765.88  580.31  772.28
#Mann= 3 , 0 , 0
       0      .1       0  421.13      .1       0  528.26      .1       0
Bank Sta=421.13,528.26
XS Rating Curve= 0 ,0
Exp/Cntr=0.3,0.1

Type RM Length L Ch R = 1 ,6583.68 ,118.89,91.44,84.4
XS GIS Cut Line= 6
     634501.6765     4314640.298     634419.6745    4315102.0982
     634425.1734    4315106.4638     634425.1734    4315123.8106
     634420.1541    4315134.5263     634415.8617    4315178.1655
#Sta/Elev= 30
       0  764.41    9.21  761.62   30.69  753.33   64.45  744.15   95.14     739
  150.39  735.05  245.53   731.2  267.01  727.24  276.22  725.93  294.63  727.71
  319.19  727.56  334.53  725.33  352.95  725.84  362.15  727.18  386.71  729.01
  398.98  727.97  408.19  725.64  414.33  725.39  429.67  727.79  441.95  728.66
  457.29  728.37  484.73   726.3  511.08  727.37  516.93  729.61  519.85  731.83
  522.77  734.94  534.47  750.93  537.39  753.71  540.31  754.02  549.08  762.79
#Mann= 3 , 0 , 0
       0      .1       0  267.01      .1       0  362.15      .1       0
Bank Sta=267.01,362.15
XS Rating Curve= 0 ,0
Exp/Cntr=0.3,0.1

Type RM Length L Ch R = 1 ,6492.24 ,109.62,91.44,74
XS GIS Cut Line= 6
     634358.8013    4314613.3104     634331.9509     4315079.904
     634335.4901    4315083.7301      634336.192    4315102.4483
     634337.8246    4315110.8603     634347.0417    4315183.2474
#Sta/Elev= 30
       0  765.66   12.22  759.92    33.6  754.05   54.98  744.69   58.04  744.63
   70.26  741.29  113.02  736.38  152.73  734.11  174.12     731  247.43  727.51
  256.59  725.94   262.7  724.65  277.98  725.82  290.19  724.32  305.47  725.39
  351.29  726.04  369.62  723.99  375.73  724.51  378.78  725.56  384.89  726.77
  397.11  727.18  512.04  725.34  527.24  726.19  530.28   727.3  536.36  732.05
   539.4   732.4  542.45  734.54  563.73  757.43  569.81  760.26  572.85  763.07
#Mann= 3 , 0 , 0
       0      .1       0  256.59      .1       0  378.78      .1       0
Bank Sta=256.59,378.78
XS Rating Curve= 0 ,0
Exp/Cntr=0.3,0.1

Type RM Length L Ch R = 1 ,6400.8  ,85.77,91.44,103.5
XS GIS Cut Line= 6
     634249.2635    4314619.6604     634242.2252    4315119.7997
     634258.8607    4315137.9649     634265.0697    4315139.9398
     634272.4516    4315151.3698     634282.2655    4315200.4804
#Sta/Elev= 30
       0  763.39    6.14  762.01   30.69  751.11   36.82  750.04   61.37  740.92
   73.65  737.61  122.75  733.73  199.46  730.22   205.6  729.28  214.81  725.54
  220.94  724.42  230.15  724.11  239.35  722.84  257.77  724.04  291.52  724.19
  300.73  723.03  309.93  723.63  343.69  723.24  349.83     724  429.61  724.74
  522.08  724.16   542.5  724.83  545.22  725.38  548.17  727.42  551.11  730.75
  554.06  731.05  565.84  747.43  574.68  756.48  580.57  760.44   595.3  765.86
#Mann= 3 , 0 , 0
       0      .1       0  230.15      .1       0  349.83      .1       0
Bank Sta=230.15,349.83
XS Rating Curve= 0 ,0
Exp/Cntr=0.3,0.1

Type RM Length L Ch R = 1 ,6309.36 ,93.97,91.44,91.2
XS GIS Cut Line= 4
     634196.8759    4314641.8855     634170.9234    4315151.4373
     634170.5377     4315163.011     634193.3041    4315304.1389
#Sta/Elev= 30
       0  755.79   18.44  748.25   24.59  747.35    46.1  741.59   61.47   739.1
  107.57   734.6  144.46  732.81  147.53  731.78  156.75  724.48  159.83  723.59
  193.63  724.52  202.86  723.36     209  722.28  242.81   723.3  255.11  722.05
  270.47  724.14  307.36  721.41   313.5   722.2  374.98  723.29  494.84  722.84
     516   724.3  543.08  730.31  564.37  732.82  579.58  736.87  597.83  737.72
  616.08  740.05  640.41  747.32  649.54  751.52  652.58  751.66  664.74  757.39
#Mann= 3 , 0 , 0
       0      .1       0  202.86      .1       0   313.5      .1       0
Bank Sta=202.86,313.5
XS Rating Curve= 0 ,0
Exp/Cntr=0.3,0.1

Type RM Length L Ch R = 1 ,6217.92 ,90.03,91.44,96.38
XS GIS Cut Line= 4
     634080.9882    4314622.8355     634080.8962    4315150.0914
     634080.2865    4315161.3056     634080.9566    4315223.3696
#Sta/Elev= 30
       0  756.84    6.13  754.51   21.46  751.23   42.92   748.7   61.31  747.53
   82.77  743.74  104.22  742.19  147.14  741.44  162.47  738.77  199.25  737.11
  205.38  734.36  208.45  734.06  220.71  724.67  226.84  721.78   248.3  721.73
  254.43  720.94  263.63  721.98  297.35  721.84  318.81  719.69  331.07  722.12
  423.03  722.74  518.06  721.64  547.35  723.22  553.26  725.39  556.22  728.54
  565.09  740.08  568.04  740.24  591.69  753.42  594.64  753.82  600.55  756.55
#Mann= 3 , 0 , 0
       0      .1       0  297.35      .1       0  331.07      .1       0
Bank Sta=297.35,331.07
XS Rating Curve= 0 ,0
Exp/Cntr=0.3,0.1

Type RM Length L Ch R = 1 ,6126.48 ,90.9,91.44,88.12
XS GIS Cut Line= 6
     634007.2796    4314653.9902     633991.5298    4315106.2455
     633990.9405    4315136.0242     633989.8027    4315154.8954
      633988.833    4315164.4166     633985.5065    4315245.1435
#Sta/Elev= 30
       0  746.08   12.23  744.66   18.35  742.97   27.52  739.18   36.69  737.93
   73.38   737.1  110.07  733.94  131.48  732.96  137.59  733.42  140.65  734.54
  162.05  736.27  174.28  731.05   201.8  726.84  226.26  720.76  232.38  720.25
   259.9  720.69  266.01  719.44  287.42  719.37  299.65  720.62  421.95  721.78
   489.3  719.99  540.72  722.02   546.7   724.2   549.7  724.45  558.67     731
  573.64  740.48  576.63  741.97  579.62  742.11  582.61  743.26  591.59  747.91
#Mann= 3 , 0 , 0
       0      .1       0   259.9      .1       0  299.65      .1       0
Bank Sta=259.9,299.65
XS Rating Curve= 0 ,0
Exp/Cntr=0.3,0.1

Type RM Length L Ch R = 1 ,6035.04 ,92.82,91.44,84.13
XS GIS Cut Line= 6
     633910.7064    4314762.4696     633905.6424     4315103.147
     633898.3428    4315145.1197     633901.1026    4315155.1075
     633901.1026    4315185.6669      633924.166     4315278.685
#Sta/Elev= 30
       0  745.92    6.14  745.01    30.7  737.02   42.97  735.03   76.74  732.32
   95.15  731.62   98.22  730.53  113.57  720.32  116.64  719.59   141.2  719.08
  153.48  718.22  174.96   719.7  227.14  719.37  236.35  718.36  257.84  719.26
  310.02  717.22   322.3   717.8  328.44  719.31  337.65  720.55  343.76   720.7
  371.15  718.66  399.79   718.5  433.22   720.3  484.14  720.49  487.13  721.45
  490.13  723.61  499.11  731.33  511.09  742.52  514.08  743.24  520.07  747.77
#Mann= 3 , 0 , 0
       0      .1       0  227.14      .1       0  328.44      .1       0
Bank Sta=227.14,328.44
XS Rating Curve= 0 ,0
Exp/Cntr=0.3,0.1

Type RM Length L Ch R = 1 ,5943.6  ,96.62,91.44,101.39
XS GIS Cut Line= 6
     633831.3313    4314762.4696     633809.2192    4315128.0312
     633808.0101    4315138.0595     633807.8632    4315161.0606
     633825.7227     4315211.067     633844.6896    4315317.0288
#Sta/Elev= 30
       0  747.29   12.21  740.96   27.47  737.51   57.99  731.94    76.3  730.85
  100.71   719.6  103.77  719.04  119.02  718.82  128.18  716.44  131.23  716.29
  143.44  717.94  210.58  720.92  231.95  720.13   241.1  718.98  247.21  717.28
  268.57   716.6  326.55  717.37  335.71  718.53  347.92  718.92  384.96  716.66
  396.46  717.39  452.43  718.23  503.26  718.23  521.21  718.98  527.19  720.01
  530.18  721.46  551.11  741.46   554.1  743.78  557.09  744.42  560.08  747.35
#Mann= 3 , 0 , 0
       0      .1       0  247.21      .1       0  396.46      .1       0
Bank Sta=247.21,396.46
XS Rating Curve= 0 ,0
Exp/Cntr=0.3,0.1

Type RM Length L Ch R = 1 ,5852.16 ,94.68,91.44,90.07
XS GIS Cut Line= 4
     633751.9782    4314741.8982     633717.8919    4315137.5073
     633720.2248    4315193.0719     633737.0488    4315378.8569
#Sta/Elev= 30
       0  755.02   15.27   746.5   18.33  746.46   45.82  736.26   48.87  736.11
   82.47  726.69  103.85  718.25  109.96  717.63  122.18  718.05  131.34  715.17
  137.45   715.4  146.61  716.97  186.32  717.54  204.65  716.88  271.84  716.88
   308.5  715.28  314.61  714.47  351.26  715.47  363.48  713.76  375.69  715.82
  411.71  716.82   458.8  714.74   495.5  715.15  550.55  716.34  584.19  718.62
  593.36  721.96  614.77  739.19  617.83  741.05  620.89  741.79  639.23   755.5
#Mann= 3 , 0 , 0
       0      .1       0   308.5      .1       0   495.5      .1       0
Bank Sta=308.5,495.5
XS Rating Curve= 0 ,0
Exp/Cntr=0.3,0.1

Type RM Length L Ch R = 1 ,5760.72 ,91.64,91.44,100.07
XS GIS Cut Line= 5
     633569.3933    4314765.1154       633626.35    4315140.5474
      633626.894    4315147.7401     633624.7633    4315158.4368
     633652.7372    4315356.4604
#Sta/Elev= 30
       0  746.85   15.31  742.01   21.44  741.12   36.75  737.16   52.06  734.45
    73.5  721.62   76.56  720.08   79.62  719.72   85.75  715.42   88.81  714.25
   91.87  714.62   97.99  716.72  104.12  717.26  171.49  715.78  202.11  714.58
   211.3  713.28  220.49  714.86  293.98   713.7  318.48   714.5  376.32  714.22
  397.85  712.71  419.06   713.9  537.23  716.64  549.36  720.95  555.42  721.97
  561.48  724.11  570.57  729.23  579.66  735.64  585.72  737.83  597.84  745.71
#Mann= 3 , 0 , 0
       0      .1       0  376.32      .1       0  419.06      .1       0
Bank Sta=376.32,419.06
XS Rating Curve= 0 ,0
Exp/Cntr=0.3,0.1

Type RM Length L Ch R = 1 ,5669.28 ,96.57,91.44,82.34
XS GIS Cut Line= 4
     633492.6639    4314766.4383     633535.8152    4315138.9841
     633535.5857    4315158.0266     633549.5495    4315344.5541
#Sta/Elev= 30
       0  748.65   27.67   740.8   30.74  740.75   58.41  734.62   67.63  733.93
   86.07  729.09   92.22  728.22  116.81   720.5  135.26  717.22  172.15  712.37
  193.67  711.21  215.18  712.31  224.41   710.5  233.63  713.64  258.22  713.63
  270.52  711.83  279.74   712.9  362.74   712.4  385.92   711.8  406.35  712.41
  440.08  714.21  489.14  715.46   492.2  716.15   501.4  721.31  504.47  721.84
  513.67  726.22  544.33  732.25  562.73  739.01   565.8  739.14  581.13  745.82
#Mann= 3 , 0 , 0
       0      .1       0  362.74      .1       0  406.35      .1       0
Bank Sta=362.74,406.35
XS Rating Curve= 0 ,0
Exp/Cntr=0.3,0.1

Type RM Length L Ch R = 1 ,5577.84 ,95.49,91.44,82.71
XS GIS Cut Line= 5
     633405.3513    4314779.6675     633426.4308    4315118.9028
     633451.9442    4315177.6609     633456.0679    4315197.8168
     633466.2056    4315340.5853
#Sta/Elev= 30
       0  746.22   30.62   741.6   55.12  736.36   61.24  735.72    88.8  730.26
   97.99  729.52   113.3  726.92  119.42  726.41  162.29  718.98  199.03  714.12
  257.21   709.9  269.46  710.23  281.71  711.46  312.33  712.03  358.19   711.8
  379.54  710.84   394.8  710.11  409.83  710.76   470.2     713  476.29  715.69
  479.34  715.91  485.43  719.03  491.52  721.22   503.7  724.63  506.74  724.65
  525.02  730.39  534.15  734.12   537.2  734.22   564.6  746.21  567.65   746.5
#Mann= 3 , 0 , 0
       0      .1       0  379.54      .1       0  409.83      .1       0
Bank Sta=379.54,409.83
XS Rating Curve= 0 ,0
Exp/Cntr=0.3,0.1

Type RM Length L Ch R = 1 ,5486.4  ,81.54,91.44,107.49
XS GIS Cut Line= 6
     633361.1658    4314779.9321     633357.8191    4315200.2973
     633367.4625    4315212.3544     633370.4925    4315217.9479
     633375.8789    4315230.3064     633409.8492    4315337.6749
#Sta/Elev= 30
       0  745.45   30.68  740.78   39.89  739.82   61.37  736.24   67.51  735.68
   116.6  727.96  128.88  727.01  141.15  724.57  187.18  721.64  211.72  714.52
  239.34  711.04  257.75  710.93  266.96  709.39  294.57  710.64   398.9  711.61
   428.1  710.26  433.24  709.42  440.06  708.74  455.66  709.65  464.79  710.44
  470.88  711.82  480.01  717.32  483.05  718.47  489.14   719.5  516.53  729.56
  522.62  730.55  543.93  738.26  546.97  739.16  550.01  739.36  568.28  747.13
#Mann= 3 , 0 , 0
       0      .1       0  433.24      .1       0  455.66      .1       0
Bank Sta=433.24,455.66
XS Rating Curve= 0 ,0
Exp/Cntr=0.3,0.1
